--- hj.prj (project) ---

Proj Title=Hwajung_plan
Current Plan=p03
Default Exp/Contr=0.3,0.1
SI Units
Geom File=g01
Flow File=f06
Flow File=f01
Flow File=f02
Flow File=f03
Flow File=f04
Flow File=f05
Plan File=p03
Plan File=p02
Plan File=p01
Y Axis Title=Elevation
X Axis Title(PF)=Main Channel Distance
X Axis Title(XS)=Station
BEGIN DESCRIPTION:
°³¼öÈÄ
END DESCRIPTION:
DSS Export Rating Curves= 0
DSS Export Rating Curve Sorted= 0
DSS Export Volume Flow Curves= 0
DXF OffsetX= 0
DXF OffsetY= 0
DXF ScaleX= 1
DXF ScaleY= 10

--- hj.p03 (plan) ---

Plan Title=Plan 03
Program Version=3.13
Short Identifier=Plan 03
Geom File=g01
Flow File=f06
Subcritical Flow
K Sum by GR= 0
Std Step Tol= 0.01
Critical Tol= 0.01
Num of Std Step Trials= 20
Max Error Tol= 0.3
Flow Tol Ratio= 0.001
Split Flow NTrial= 30
Split Flow Tol= 0.02
Split Flow Ratio= 0.02
Log Output Level= 0
Friction Slope Method= 1
Unsteady Friction Slope Method= 2
Unsteady Bridges Friction Slope Method= 1
Parabolic Critical Depth
Global Vel Dist= 0 , 0 , 0
Global Log Level= 0
CheckData=True
Encroach Param=-1 ,0,0, 0
Computation Interval=1HOUR
Output Interval=1HOUR
Run HTab= 0
Run UNet= 0
Run PostProcess= 0
UNET Theta= 1
UNET Theta Warmup= 1
UNET ZTol= 0.02
UNET ZSATol= 0.05
UNET MxIter= 20
UNET MaxInSteps= 0
UNET DtIC= 0
UNET DtMin= 0
UNET MaxCRTS= 20
UNET WFStab= 2
UNET SFStab= 1
UNET WFX= 1
UNET SFX= 1
UNET DSS MLevel= 4
UNET DZMax Abort= 100
UNET Convert EG Bridges=-1
UNET Use Existing IB Tables=-1
UNET Froude Reduction=False
UNET Froude Limit= 1
UNET Froude Power= 10
Instantaneous Interval=1HOUR
DSS File=dss
Write IC File= 0
Echo Input=False
Echo Output=False
Write Detailed= 0
Detailed Automatic Start=False, 10

--- hj.p01 (plan) ---

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Plan Title=Plan 01
Short Identifier=1
Geom File=g01
Flow File=f01
Supercritical Flow

--- hj.p02 (plan) ---

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Plan Title=Plan 02
Geom File=g01

--- hj.f06 (steady flow) ---

Flow Title=plan
Program Version=3.12
Number of Profiles= 14
Profile Names=96',1.58yr,10yr,20yr,30yr,50yr,80yr,100yr,200yr,plan,PF 11,PF 12,2001yr,2006yr
River Rch & RM=RIVER-1,Reach-1         ,104
     215      35      75      90     100     110     120     125     140     125
     .23     .27      49       2
River Rch & RM=RIVER-1,Reach-1         ,87
     215      50     110     135     145     160     175     180     200     180
     .23     .27     119       3
River Rch & RM=RIVER-1,Reach-1         ,69.22
     295      65     140     165     180     200     215     225     250     225
     .23     .27     178       5
River Rch & RM=RIVER-1,Reach-1         ,30.38
     385      75     160     190     205     225     245     255     285     255
     .23     .27     207       6
Boundary for River Rch & Prof#=RIVER-1,Reach-1         , 1
Up Type= 0
Dn Type= 1
Dn Known WS=2.31
Boundary for River Rch & Prof#=RIVER-1,Reach-1         , 2
Up Type= 0
Dn Type= 1
Dn Known WS=0.24
Boundary for River Rch & Prof#=RIVER-1,Reach-1         , 3
Up Type= 0
Dn Type= 1
Dn Known WS=1.24
Boundary for River Rch & Prof#=RIVER-1,Reach-1         , 4
Up Type= 0
Dn Type= 1
Dn Known WS=1.51
Boundary for River Rch & Prof#=RIVER-1,Reach-1         , 5
Up Type= 0
Dn Type= 1
Dn Known WS=1.68
Boundary for River Rch & Prof#=RIVER-1,Reach-1         , 6
Up Type= 0
Dn Type= 1
Dn Known WS=1.86
Boundary for River Rch & Prof#=RIVER-1,Reach-1         , 7
Up Type= 0
Dn Type= 1
Dn Known WS=2.02
Boundary for River Rch & Prof#=RIVER-1,Reach-1         , 8
Up Type= 0
Dn Type= 1
Dn Known WS=2.05
Boundary for River Rch & Prof#=RIVER-1,Reach-1         , 9
Up Type= 0
Dn Type= 1
Dn Known WS=2.32
Boundary for River Rch & Prof#=RIVER-1,Reach-1         , 10
Up Type= 0
Dn Type= 1
Dn Known WS=2.05
Boundary for River Rch & Prof#=RIVER-1,Reach-1         , 11
Up Type= 0
Dn Type= 1
Dn Known WS=-1
Boundary for River Rch & Prof#=RIVER-1,Reach-1         , 12
Up Type= 0
Dn Type= 1
Dn Known WS=-1
Boundary for River Rch & Prof#=RIVER-1,Reach-1         , 13
Up Type= 0
Dn Type= 1
Dn Known WS=1.68
Boundary for River Rch & Prof#=RIVER-1,Reach-1         , 14
Up Type= 0
Dn Type= 1
Dn Known WS=-0.98
DSS Import GetInterval= 0
DSS Import GetPeak= 0
DSS Import FillOption= 0

--- hj.f01 (steady flow) ---

Flow Title=Flow 01
Program Version=3.13
Number of Profiles= 1
Profile Names=plan
River Rch & RM=RIVER-1,Reach-1         ,104
     215
River Rch & RM=RIVER-1,Reach-1         ,69.22
     295
River Rch & RM=RIVER-1,Reach-1         ,27.08
     385
Boundary for River Rch & Prof#=RIVER-1,Reach-1         , 1
Up Type= 0
Dn Type= 1
Dn Known WS=2.44
DSS Import GetInterval= 0
DSS Import GetPeak= 0
DSS Import FillOption= 0

--- hj.f02 (steady flow) ---

Flow Title=Flow 02
Program Version=3.11
Number of Profiles= 1
Profile Names=PF 1
River Rch & RM=RIVER-1,Reach-1         ,104
DSS Import GetInterval= 0
DSS Import GetPeak= 0
DSS Import FillOption= 0

--- hj.f03 (steady flow) ---

Flow Title=Flow 03
Program Version=3.13
Number of Profiles= 1
Profile Names=PF 1
DSS Import GetInterval= 0
DSS Import GetPeak= 0
DSS Import FillOption= 0

--- hj.f04 (steady flow) ---

Flow Title=Flow 04
Program Version=3.13
Number of Profiles= 1
Profile Names=96'
River Rch & RM=RIVER-1,Reach-1         ,104
     215
River Rch & RM=RIVER-1,Reach-1         ,69.21
     295
River Rch & RM=RIVER-1,Reach-1         ,30.379
     385
Boundary for River Rch & Prof#=RIVER-1,Reach-1         , 1
Up Type= 3
Up Slope=0.001999
Dn Type= 1
Dn Known WS=2.31
DSS Import GetInterval= 0
DSS Import GetPeak= 0
DSS Import FillOption= 0

--- hj.f05 (steady flow) ---

Flow Title=Flow 05
Program Version=3.13
Number of Profiles= 1
Profile Names=PF 1
River Rch & RM=RIVER-1,Reach-1         ,104
     215
River Rch & RM=RIVER-1,Reach-1         ,69
     295
River Rch & RM=RIVER-1,Reach-1         ,30
     385
Boundary for River Rch & Prof#=RIVER-1,Reach-1         , 1
Up Type= 0
Dn Type= 1
Dn Known WS=2.31
DSS Import GetInterval= 0
DSS Import GetPeak= 0
DSS Import FillOption= 0

--- hj.g01 (geometry) ---

Geom Title=Geom 01
Program Version=3.12

River Reach=RIVER-1         ,Reach-1
Reach XY= 2
              .5             .95              .5             .05

Type RM Length L Ch R = 1 ,104     ,3,3,3
#Sta/Elev= 24
       0   10.92      30   10.92      30   10.42    30.5   10.42    30.5    8.62
    32.5    7.38      41    7.38    45.5    7.38      46    6.87    46.5    6.52
    47.5    6.57    48.5    6.87      49    7.41    51.5    7.41      57   10.32
    57.5   10.42      58   10.42      58   11.42      63   11.42      63   11.22
    71.5   11.34    80.5   11.18    80.5   11.42    82.5   13.82
#Mann= 3 , 0 , 0
       0     .03       0      30     .03       0      58     .03       0
Bank Sta=30,58
Exp/Cntr=0.3,0.1

Type RM Length L Ch R = 1 ,103.47  ,20,20,20
#Sta/Elev= 17
       0   11.37    36.5   11.43    36.5   10.58    37.5   10.58    37.5    8.55
      40    7.57      55    6.76      57    6.56      58    6.56    58.5    6.76
      67    7.22    68.5     8.5    68.5   10.58    69.5   10.58    69.5   11.43
      72   11.47     100   12.52
#Mann= 3 , 0 , 0
       0     .03       0    36.5     .03       0    69.5     .03       0
Bank Sta=36.5,69.5
Exp/Cntr=0.5,0.3

Type RM Length L Ch R = 3 ,103.37  ,,,
BEGIN DESCRIPTION:
È­Á¤8±³
END DESCRIPTION:
Bridge Culvert--1,0,-1,-1, 0
Deck Dist Width WeirC Skew NumUp NumDn MinLoCord MaxHiCord MaxSubmerge Is_Ogee
0.1,19,1.44,0, 2, 2, , , 0.95, 0, 0,0,,
    36.5    69.5
   11.43   11.43
   10.58   10.58
    36.5    69.5
   11.43   11.43
   10.58   10.58
Pier Skew, UpSta & Num, DnSta & Num=  ,54.5, 2 ,54.5, 2 , 0 , 0 , 0 ,,
      .7      .7
       5      11
      .7      .7
       5      11
BR Coef=-1 , 0 , 0 ,, 0 ,,,0.8,-1,,0,
WSPro=,,,, 1 ,,,, 0 ,,,, 0 ,,,,-1 ,-1 ,-1 , 0 , 0 , 0 , 0 , 0
BC Design=,, 0 ,, 0 ,,,,,,

Type RM Length L Ch R = 1 ,103.27  ,27,27,27
#Sta/Elev= 17
       0   11.37    36.5   11.43    36.5   10.58    37.5   10.58    37.5    8.55
      40    7.57      55    6.76      57    6.56      58    6.56    58.5    6.76
      67    7.22    68.5     8.5    68.5   10.58    69.5   10.58    69.5   11.43
      72   11.47     100   12.52
#Mann= 3 , 0 , 0
       0     .03       0    36.5     .03       0    69.5     .03       0
Bank Sta=36.5,69.5
Exp/Cntr=0.5,0.3

Type RM Length L Ch R = 1 ,103     ,50,50,50
#Sta/Elev= 30
       0   11.28       9   11.28       9   12.38    20.6   13.49    28.2    13.7
    37.5   13.47      48   10.44    50.6   10.34    50.6   10.14    57.5   10.37
    64.1   10.04    64.5   10.04    64.5   10.24   72.33   10.24   72.47   10.24
      74    7.46    75.5     7.3    80.5    7.29      81    6.87    83.5     6.9
    84.5    6.64      89    7.27    92.5    7.32    97.7    9.98    97.7   11.38
      98   11.38     101   11.38     101   11.18   146.5   13.83     169   16.18
#Mann= 3 , 0 , 0
       0     .03       0   72.33     .03       0      98     .03       0
Bank Sta=72.33,98
Exp/Cntr=0.3,0.1

Type RM Length L Ch R = 1 ,102     ,13,13,13
#Sta/Elev= 30
       0   11.13    39.4   11.15    39.4    10.9    58.7   10.81    58.7   11.06
    61.7   11.21    61.7    9.86    66.2    7.69    68.7    7.38    73.2    7.36
    75.2    6.71    76.2    6.61    77.2    6.71    79.7    7.38    84.5    7.36
    86.2    7.46    89.4    8.97    91.4    9.71    91.4   11.06    92.2   11.06
    94.4   11.06    94.4   10.86   101.7   10.91   108.7    10.7   108.7    10.9
   111.7   11.16   111.7   12.16   128.7   14.33   137.9   14.19   167.9   14.19
#Mann= 3 , 0 , 0
       0     .03       0    61.7     .03       0    92.2     .03       0
Bank Sta=61.7,92.2
Exp/Cntr=0.3,0.1

Type RM Length L Ch R = 1 ,101.37  ,17,17,17
#Sta/Elev= 21
       0   10.94      40   10.94      40   10.04      41   10.04      41    8.24
    43.5    7.29      50    7.24    50.5    6.62      53    6.52      56    6.52
    56.5    6.52      62    6.52    62.5    6.62      63    7.64      70    7.74
      71    8.74      71   10.04      72   10.04      72   10.94    73.5   10.94
     110   10.94
#Mann= 3 , 0 , 0
       0     .03       0      40     .03       0    73.5     .03       0
Bank Sta=40,73.5
Exp/Cntr=0.5,0.3

Type RM Length L Ch R = 3 ,101.285 ,,,
BEGIN DESCRIPTION:
È­Á¤7±³
END DESCRIPTION:
Bridge Culvert--1,0,-1,-1, 0
Deck Dist Width WeirC Skew NumUp NumDn MinLoCord MaxHiCord MaxSubmerge Is_Ogee
0.1,16,1.44,0, 2, 2, , , 0.95, 0, 0,0,,
      40    73.5
   10.94   10.94
   10.04   10.04
      40    73.5
   10.94   10.94
   10.04   10.04
Pier Skew, UpSta & Num, DnSta & Num=  ,56, 2 ,56, 2 , 0 , 0 , 0 ,,
      .6      .6
       5      11
      .6      .6
       5      11
BR Coef=-1 , 0 , 0 ,, 0 ,,,0.8,-1,,0,
WSPro=,,,, 1 ,,,, 0 ,,,, 0 ,,,,-1 ,-1 ,-1 , 0 , 0 , 0 , 0 , 0
BC Design=,, 0 ,, 0 ,,,,,,

Type RM Length L Ch R = 1 ,101.20  ,20,20,20
#Sta/Elev= 21
       0   10.94      40   10.94      40   10.04      41   10.04      41    8.24
    43.5    7.29      50    7.24    50.5    6.62      53    6.52      56    6.52
    56.5    6.52      62    6.52    62.5    6.62      63    7.64      70    7.74
      71    8.74      71   10.04      72   10.04      72   10.94    73.5   10.94
     110   10.94
#Mann= 3 , 0 , 0
       0     .03       0      40     .03       0    73.5     .03       0
Bank Sta=40,73.5
Exp/Cntr=0.5,0.3

Type RM Length L Ch R = 1 ,101     ,50,50,50
#Sta/Elev= 28
       0   10.72      33   10.72      33   10.92    33.5   10.92      40   10.65
      47   10.52      47   10.72    50.5   10.81    50.5    9.78      55     7.4
    60.5    7.34    60.5    6.62    61.5     6.5      62    6.35      65    6.35
    65.5     6.5    69.8     6.8    70.5    7.34    73.5    7.29      76    7.48
    80.3    9.42    80.3   10.92      82   10.92    83.2   10.72    90.3   10.86
    97.5   10.65   103.5   11.19   133.5   11.19
#Mann= 3 , 0 , 0
       0     .03       0    50.5     .03       0      82     .03       0
Bank Sta=50.5,82
Exp/Cntr=0.3,0.1

Type RM Length L Ch R = 1 ,100     ,50,50,50
#Sta/Elev= 24
       0    9.38     5.4    9.56    11.9    9.48    12.4    9.48    12.4    9.68
    15.4    9.61    15.4    9.41    16.4    8.93    19.9    7.22   20.23    7.06
    26.4    7.06    28.8    5.86    31.8    5.86    35.4    7.06   40.38    7.06
    40.6    7.17    45.2    9.44    45.2    9.79    47.1    9.79    48.3    9.79
    48.3    9.59    48.8    9.59    55.5    9.76      60    9.61
#Mann= 3 , 0 , 0
       0     .03       0    15.4     .03       0    45.2     .03       0
Levee=-1,15.4,9.61,-1,45.2,9.79,,
Bank Sta=15.4,45.2
Exp/Cntr=0.3,0.1

Type RM Length L Ch R = 1 ,99      ,50,50,50
#Sta/Elev= 22
       0     8.9     5.4    9.02    11.7    9.05    12.2    9.05    12.2    9.25
    15.2    9.25    16.8    8.59    19.7    7.19   20.28    6.91   27.65    6.91
   30.05    5.71   33.05    5.71   36.65    6.91   40.19    6.91    40.4    7.02
    45.2    9.44    47.1    9.44    48.3    9.44    48.3    9.24    48.8    9.24
    55.3    9.31      60    9.19
#Mann= 3 , 0 , 0
       0     .03       0    15.2     .03       0    45.2     .03       0
Levee=-1,15.2,9.25,-1,45.2,9.44,,
Bank Sta=15.2,45.2
Exp/Cntr=0.3,0.1

Type RM Length L Ch R = 1 ,98      ,50,50,50
#Sta/Elev= 23
       0     8.9       5    8.87    11.6    8.76    12.1    8.76    12.1    8.96
    15.1    8.96    16.9    8.41    20.1    6.97   20.56    6.77   26.59    6.77
   28.99    5.57   31.99    5.57   35.59    6.77    44.1    6.77    44.1    6.82
    44.1    9.02    45.1    9.32    47.1    9.32    48.3    9.32    48.3    9.12
    48.8    9.12    55.3    9.21      60    9.18
#Mann= 3 , 0 , 0
       0     .03       0    15.1     .03       0    45.1     .03       0
Levee=-1,15.1,8.96,-1,45.1,9.32,,
Bank Sta=15.1,45.1
Exp/Cntr=0.3,0.1

Type RM Length L Ch R = 1 ,97      ,50,50,50
#Sta/Elev= 22
       0    8.52     5.1    8.68    11.6    8.44    12.1    8.44    12.1    8.64
    15.1    8.56    16.9    8.14    20.3    6.74    20.6    6.62   25.54    6.62
   27.94    5.42   30.94    5.42   34.54    6.62   40.03    6.62    40.2     6.7
    45.3    9.08    47.1    9.08    48.3    9.08    48.3    8.88    48.8    8.88
    55.3    8.94      60    8.85
#Mann= 3 , 0 , 0
       0     .03       0    12.1     .03       0    45.3     .03       0
Levee=-1,12.1,9,-1,45.3,9.08,,
Bank Sta=12.1,45.3
Exp/Cntr=0.3,0.1

Type RM Length L Ch R = 1 ,96      ,50,50,50
#Sta/Elev= 23
       0    8.43     5.5    8.61    11.8    8.25    12.3    8.25    12.3    8.75
    15.3    8.75    17.1    8.14    20.4    6.77   21.12    6.47    26.7    6.47
    29.1    5.27    32.1    5.27    35.7    6.47    39.8    6.47    40.4    6.76
    43.6     8.3    45.3    8.98    47.1    8.98    48.3    8.98    48.3    8.78
    48.8    8.78    55.8    8.81      60    8.72
#Mann= 3 , 0 , 0
       0     .03       0    15.3     .03       0    45.3     .03       0
Levee=-1,15.3,8.75,-1,45.3,8.98,,
Bank Sta=15.3,45.3
Exp/Cntr=0.3,0.1

Type RM Length L Ch R = 1 ,95      ,25,25,25
#Sta/Elev= 25
       0    9.13     5.2    9.26    11.8    9.12    12.3    9.12    12.3    9.32
    15.3    9.41    15.3    8.71    19.2     8.6    20.6    7.08    21.3    6.32
   25.76    6.32   28.16    5.12   31.16    5.12   34.76    6.32   38.41    6.32
    38.7    6.56    41.3    8.63    45.3    8.63    45.3    9.43    47.1    9.43
    48.3    9.43    48.3    9.23    48.8    9.23    55.4    9.33      60    9.24
#Mann= 3 , 0 , 0
       0     .03       0    15.3     .03       0    45.3     .03       0
Levee=-1,15.3,9.41,-1,45.3,9.43,,
Bank Sta=15.3,45.3
Exp/Cntr=0.3,0.1

Type RM Length L Ch R = 1 ,94.25   ,17,17,17
#Sta/Elev= 18
       0    9.45   19.35    9.59   19.35    8.94   20.35    8.94   20.35    7.55
    22.6     6.2   28.21     6.2   30.61       5   36.81       5   39.21     6.2
   42.95     6.2   44.35     6.9   44.35    8.94   45.35    8.94   45.35    9.59
   48.85    9.59   59.35     9.3      60    9.31
#Mann= 3 , 0 , 0
       0     .03       0   19.35     .03       0   45.35     .03       0
Bank Sta=19.35,45.35
Exp/Cntr=0.5,0.3

Type RM Length L Ch R = 3 ,94.165  ,,,
BEGIN DESCRIPTION:
È­Á¤6±³
END DESCRIPTION:
Bridge Culvert--1,0,-1,-1, 0
Deck Dist Width WeirC Skew NumUp NumDn MinLoCord MaxHiCord MaxSubmerge Is_Ogee
0.1,15,1.44,0, 2, 2, , , 0.95, 0, 0,0,,
   19.35   45.35
    9.59    9.59
    8.94    8.94
   19.35   45.35
    9.59    9.59
    8.94    8.94
Pier Skew, UpSta & Num, DnSta & Num=  ,31.87, 2 ,31.87, 2 , 0 , 0 , 0 ,,
      .6      .6
       5      10
      .6      .6
       5      10
BR Coef=-1 , 0 , 0 ,, 0 ,,,0.8,-1,,0,
WSPro=,,,, 1 ,,,, 0 ,,,, 0 ,,,,-1 ,-1 ,-1 , 0 , 0 , 0 , 0 , 0
BC Design=,, 0 ,, 0 ,,,,,,

Type RM Length L Ch R = 1 ,94.08   ,8,8,8
#Sta/Elev= 18
       0    9.45   19.35    9.59   19.35    8.94   20.35    8.94   20.35    7.55
    22.6     6.2   28.21     6.2   30.61       5   36.81       5   39.21     6.2
   42.95     6.2   44.35     6.9   44.35    8.94   45.35    8.94   45.35    9.59
   48.85    9.59   59.35     9.3      60    9.31
#Mann= 3 , 0 , 0
       0     .03       0   19.35     .03       0   45.35     .03       0
Bank Sta=19.35,45.35
Exp/Cntr=0.5,0.3

Type RM Length L Ch R = 1 ,94      ,50,50,50
#Sta/Elev= 24
       0    9.55     5.1    9.57    12.1    9.31    12.6    9.31    12.6    9.51
    15.4    9.81    15.4    8.89    19.8    6.97   21.62    6.18   27.89    6.18
   30.29    4.98   33.29    4.98   36.89    6.18   39.24    6.18    40.5    6.77
    44.8    8.79    45.3    8.79    45.3    9.79    47.1    9.79    48.6    9.62
    48.6    9.42    49.1    9.42    55.5    9.49      60    9.33
#Mann= 3 , 0 , 0
       0     .03       0    15.4     .03       0    45.3     .03       0
Levee=-1,15.4,9.81,-1,45.3,9.79,,
Bank Sta=15.4,45.3
Exp/Cntr=0.3,0.1

Type RM Length L Ch R = 1 ,93      ,50,50,50
#Sta/Elev= 22
       0    8.43     5.3    8.64    11.9    8.37    12.4    8.37    12.4    8.47
    15.4    8.71    20.6    6.49   21.67    6.03   28.15    6.03   30.55    4.83
   33.55    4.83   37.15    6.03    38.7    6.03    40.6    6.61    45.5     8.1
    46.2     8.1    46.2     8.3    47.1     8.3    48.4    8.49    48.9    8.49
    55.3    8.75      60    8.61
#Mann= 3 , 0 , 0
       0     .03       0    15.4     .03       0    55.3     .03       0
Levee=-1,15.4,8.71,-1,55.3,8.75,,
Bank Sta=15.4,55.3
Exp/Cntr=0.3,0.1

Type RM Length L Ch R = 1 ,92      ,50,50,50
#Sta/Elev= 21
       0    8.47     5.4    8.64    11.9    8.35    12.4    8.35    15.4    8.69
    16.2    8.47    20.9    6.42   22.13    5.89   27.63    5.89   30.03    4.69
   33.03    4.69   36.63    5.89   39.06    5.89    40.1    6.33    45.3    8.55
    47.1    8.55    48.3    8.55    48.3    8.45    48.8    8.45    55.4    8.62
      60     8.5
#Mann= 3 , 0 , 0
       0     .03       0    15.4     .03       0    45.3     .03       0
Levee=-1,15.4,8.69,-1,45.3,8.55,,
Bank Sta=15.4,45.3
Exp/Cntr=0.3,0.1

Type RM Length L Ch R = 1 ,91      ,50,50,50
#Sta/Elev= 20
       0    8.35     5.4    8.35      12     8.2    12.5     8.2    16.1    8.35
    17.6     7.6    20.6     6.2   21.59    5.74   27.86    5.74   30.26    4.54
   33.26    4.54   36.86    5.74   39.26    5.74    40.3     6.2    45.5     8.5
    47.1     8.5    48.5    8.37      49    8.37    55.5    8.55      60    8.49
#Mann= 3 , 0 , 0
       0     .03       0    16.1     .03       0    45.5     .03       0
Levee=-1,16.1,8.35,-1,45.5,8.5,,
Bank Sta=16.1,45.5
Exp/Cntr=0.3,0.1

Type RM Length L Ch R = 1 ,90      ,50,50,50
#Sta/Elev= 22
       0    8.07     .19    8.07    6.79    8.22   13.29    8.02   13.79    8.02
   16.79    8.22   16.79    8.02   17.59    8.02   21.89    6.27   23.54     5.6
   29.61     5.6   32.01     4.4   35.01     4.4   38.61     5.6   40.89     5.6
   42.09    6.21   46.79    8.62   48.49    8.52   49.79    8.31   50.29    8.31
   56.69    8.54      60    8.43
#Mann= 3 , 0 , 0
       0     .03       0   16.79     .03       0   46.79     .03       0
Levee=-1,16.79,8.22,-1,46.79,8.62,,
Bank Sta=16.79,46.79
Exp/Cntr=0.3,0.1

Type RM Length L Ch R = 1 ,89      ,50,50,50
#Sta/Elev= 21
       0    8.08    6.89    8.22   13.29    8.07   13.79    8.07   16.79    8.22
   17.29    8.32   18.19    7.72   22.69    5.87    23.7    5.45   29.67    5.45
   32.07    4.25   35.07    4.25   38.67    5.45   40.77    5.45   41.79    5.97
   46.69    8.47   48.49    8.42   49.69    8.37   50.19    8.37   56.69    8.47
      60     8.4
#Mann= 3 , 0 , 0
       0     .03       0   17.29     .03       0   46.69     .03       0
Levee=-1,17.29,8.32,-1,46.69,8.47,,
Bank Sta=17.29,46.69
Exp/Cntr=0.3,0.1

Type RM Length L Ch R = 1 ,88      ,30,30,30
#Sta/Elev= 23
       0    8.52     .29    8.52    6.89    8.62   13.39    8.42   13.89    8.42
   16.89    8.72   16.89    8.07   17.89    7.82   22.19    5.72   23.04     5.3
   27.65    5.31   30.05    4.11   33.05    4.11   36.65    5.31   40.38     5.3
   40.89    5.52   46.79    8.02   46.79    8.72   48.49    8.62   49.79    8.46
   50.29    8.46   56.79    8.61      60    8.54
#Mann= 3 , 0 , 0
       0     .03       0   16.89     .03       0   46.79     .03       0
Levee=-1,16.89,8.72,-1,46.79,8.72,,
Bank Sta=16.89,46.79
Exp/Cntr=0.3,0.1

Type RM Length L Ch R = 1 ,87.20   ,20,20,20
#Sta/Elev= 19
       0    9.14   18.99    9.08   18.99    8.43   19.99    8.43   19.99    6.68
   22.99    5.18   23.03    5.16   27.83    5.16   30.23    3.96   36.05    3.96
   38.45    5.16   42.12    5.16   42.49    5.38   43.99    6.28   43.99    8.37
   44.99    8.37   44.99    9.02   48.49    9.05      60    9.06
#Mann= 3 , 0 , 0
       0     .03       0   18.99     .03       0   44.99     .03       0
Levee=-1,18.99,9.08,-1,44.99,9.02,,
Bank Sta=18.99,44.99
Exp/Cntr=0.5,0.3

Type RM Length L Ch R = 3 ,87.10   ,,,
BEGIN DESCRIPTION:
È­Á¤5±³
END DESCRIPTION:
Bridge Culvert--1,0,-1,-1, 0
Deck Dist Width WeirC Skew NumUp NumDn MinLoCord MaxHiCord MaxSubmerge Is_Ogee
0.1,19,1.44,0, 2, 2, , , 0.95, 0, 0,0,,
   18.99   44.99
    9.08    9.02
    8.43    8.37
   18.99   44.99
    9.08    9.02
    8.43    8.37
Pier Skew, UpSta & Num, DnSta & Num=  ,32, 2 ,32, 2 , 0 , 0 , 0 ,,
      .6      .6
       4     9.5
      .6      .6
       4     9.5
BR Coef=-1 , 0 , 0 ,, 0 ,,,0.8,-1,,0,
WSPro=,,,, 1 ,,,, 0 ,,,, 0 ,,,,-1 ,-1 ,-1 , 0 , 0 , 0 , 0 , 0
BC Design=,, 0 ,, 0 ,,,,,,

Type RM Length L Ch R = 1 ,87      ,50,50,50
#Sta/Elev= 19
       0    9.14   18.99    9.08   18.99    8.43   19.99    8.43   19.99    6.68
   22.99    5.18   23.03    5.16   27.83    5.16   30.23    3.96   36.05    3.96
   38.45    5.16   42.12    5.16   42.49    5.38   43.99    6.28   43.99    8.37
   44.99    8.37   44.99    9.02   48.49    9.05      60    9.06
#Mann= 3 , 0 , 0
       0     .03       0   18.99     .03       0   44.99     .03       0
Levee=-1,18.99,9.08,-1,44.99,9.02,,
Bank Sta=18.99,44.99
Exp/Cntr=0.5,0.3

Type RM Length L Ch R = 1 ,86      ,50,50,50
#Sta/Elev= 22
       0    7.95     .09    7.95    6.49    8.25   13.39       8   13.89       8
   13.89     8.3   16.89     8.3   21.69     5.8   23.07    5.08   27.34    5.08
   29.74    3.88   33.74    3.88   37.34    5.08   41.08    5.08   41.89    5.55
   46.89     8.5   48.49     8.5   49.89     8.4   49.89     8.2   50.39     8.2
   56.99    8.34      60    8.37
#Mann= 3 , 0 , 0
       0     .03       0   16.89     .03       0   46.89     .03       0
Levee=-1,16.89,8.3,-1,46.89,8.5,,
Bank Sta=16.89,46.89
Exp/Cntr=0.3,0.1

Type RM Length L Ch R = 1 ,85      ,50,50,50
#Sta/Elev= 23
       0    8.02     .49    8.02    6.69    8.17   13.49    7.97   13.99    7.97
   15.49    8.12   15.49    8.22   16.99    8.22   22.19    5.72    23.7    4.99
   28.03    4.99   30.43    3.79   34.43    3.79   38.03    4.99   40.55    4.99
   41.49    5.47   46.89    8.22   48.49    8.22   49.89    8.12   49.89    7.92
   50.39    7.92   56.79    8.13      60     8.1
#Mann= 3 , 0 , 0
       0     .03       0   16.99     .03       0   46.89     .03       0
Levee=-1,16.99,8.22,-1,46.89,8.22,,
Bank Sta=16.99,46.89
Exp/Cntr=0.3,0.1

Type RM Length L Ch R = 1 ,84      ,50,50,50
#Sta/Elev= 24
       0    7.96     .19    7.96    6.59    8.12   13.59       8   14.09       8
   15.59    8.16   15.59    8.26   17.09    8.26   18.59    7.44   22.69    5.59
   24.19    4.91   28.58    4.91   30.98    3.71   34.98    3.71   38.58    4.91
   39.99    4.91   40.79    5.28   46.99    8.14   48.49    8.14   49.99    8.04
   49.99    7.84   50.49    7.84   56.99    8.04      60       8
#Mann= 3 , 0 , 0
       0     .03       0   17.09     .03       0   46.99     .03       0
Levee=-1,17.09,8.26,-1,46.99,8.14,,
Bank Sta=17.09,46.99
Exp/Cntr=0.3,0.1

Type RM Length L Ch R = 1 ,83      ,50,50,50
#Sta/Elev= 24
       0    8.06    4.99    8.14   11.69    7.94   12.19    7.94   13.99    8.14
   13.99    8.24   15.49    8.24   16.79    7.49   21.89    5.25   22.85    4.83
   27.26    4.83   29.66    3.63   33.66    3.63   37.26    4.83   39.25    4.83
   40.19    5.25   45.09    7.47   46.99    8.24   48.49    8.24   49.99    8.14
   49.99    7.94   50.49    7.94   56.99    8.12      60    8.05
#Mann= 3 , 0 , 0
       0     .03       0   15.49     .03       0   46.99     .03       0
Levee=-1,15.49,8.24,-1,46.99,8.24,,
Bank Sta=15.49,46.99
Exp/Cntr=0.3,0.1

Type RM Length L Ch R = 1 ,82      ,50,50,50
#Sta/Elev= 22
       0    8.04    6.49    7.91    6.99    7.91    8.49    8.02    9.99    8.12
   10.99    7.55   15.39    5.36   16.62    4.74   26.54    4.75   28.94    3.54
   32.94    3.54   36.54    4.75   41.33    4.74   42.69    5.41   46.69    7.37
   48.29    8.19   50.49    8.19   51.29    8.19   51.29    7.99   51.79    7.99
   58.19    8.13      60     8.1
#Mann= 3 , 0 , 0
       0     .03       0    9.99     .03       0   48.29     .03       0
Bank Sta=9.99,48.29
Exp/Cntr=0.3,0.1

Type RM Length L Ch R = 1 ,81      ,50,50,50
#Sta/Elev= 23
       0    7.97    4.99    7.83    5.49    7.83    6.99    7.87    6.99    8.07
    8.59    8.07    9.99    7.56   14.69     5.2   15.76    4.66      25    4.66
    27.4    3.46    31.4    3.46      35    4.66   41.14    4.66   42.59    5.33
   46.99    7.36   48.49    8.14   50.49    8.14   51.49    8.14   51.49    7.94
   51.99    7.94   58.49    8.24      60     8.2
#Mann= 3 , 0 , 0
       0     .03       0    8.59     .03       0   48.49     .03       0
Levee=-1,8.59,8.07,-1,48.49,8.14,,
Bank Sta=8.59,48.49
Exp/Cntr=0.3,0.1

Type RM Length L Ch R = 1 ,80      ,50,50,50
#Sta/Elev= 22
       0    7.92    4.29     7.8    4.79     7.8    6.29    8.01    7.69    8.16
    9.19     7.6   14.59    5.15   15.84    4.58   23.18    4.58   25.58    3.38
   29.58    3.38   33.18    4.58   40.82    4.58   42.39    5.34   46.09    7.14
   47.69    8.13   50.49    8.03   50.69    8.03   50.69    7.83   51.19    7.83
   57.79    8.14      60    8.08
#Mann= 3 , 0 , 0
       0     .03       0    7.69     .03       0   47.69     .03       0
Bank Sta=7.69,47.69
Exp/Cntr=0.3,0.1

Type RM Length L Ch R = 1 ,79      ,50,50,50
#Sta/Elev= 24
       0    7.99    5.49    7.77    6.69    7.77    7.19    7.98    7.19    8.08
    8.49    8.08    9.69    8.16   11.29    7.36   16.49    4.99   17.57     4.5
   27.57     4.5   29.97     3.3   33.97     3.3   37.57     4.5    42.5     4.5
   44.19    5.19   47.39    6.51   50.09    7.93   50.49    7.93   53.09    7.93
   53.09    7.73   53.59    7.73   59.99    7.78      60    7.78
#Mann= 3 , 0 , 0
       0     .03       0    9.69     .03       0   50.09     .03       0
Levee=-1,9.69,8.16,-1,50.09,7.93,,
Bank Sta=9.69,50.09
Exp/Cntr=0.3,0.1

Type RM Length L Ch R = 1 ,78      ,50,50,50
#Sta/Elev= 22
       0    8.12    5.09     7.9    5.49     7.9    5.49    8.05    8.49     8.1
    9.69    7.44   14.89    4.94   15.98    4.41   28.31    4.41   30.71    3.21
   34.71    3.21   38.31    4.41   40.99    4.41   41.79    4.76   46.19    6.69
   48.49    7.83   49.99    7.83   51.49    7.83   51.49    7.63   51.99    7.63
   58.39    7.79      60    7.76
#Mann= 3 , 0 , 0
       0     .03       0    8.49     .03       0   48.49     .03       0
Bank Sta=8.49,48.49
Exp/Cntr=0.3,0.1

Type RM Length L Ch R = 1 ,77      ,10,10,10
#Sta/Elev= 24
       0    8.64    5.09    8.46    5.59    8.46    5.59    8.66    8.79    8.71
    8.79    7.71    9.69    7.41   14.89     4.9   16.07    4.33   27.19    4.33
   29.59    3.13   33.59    3.13   37.19    4.33   41.21    4.33   42.09    4.74
   45.79    6.47   48.69    7.78   48.69    8.28   49.99    8.28   51.69    8.28
   51.69    8.08   52.19    8.08   58.49    8.27      60    8.22
#Mann= 3 , 0 , 0
       0     .03       0    8.79     .03       0   48.69     .03       0
Levee=-1,8.79,8.71,-1,48.69,8.28,,
Bank Sta=8.79,48.69
Exp/Cntr=0.3,0.1

Type RM Length L Ch R = 1 ,76.40   ,20,20,20
#Sta/Elev= 19
       0    8.49    5.59    8.47    5.59    7.17    6.59    7.17    6.59    5.86
   10.59    4.46    11.1    4.28   23.33    4.28   25.73    3.08   31.83    3.08
   34.23    4.28   42.73    4.28   43.29    4.56   45.29    5.56   45.29    7.18
   46.29    7.18   46.29    8.48   49.99    8.48      60    8.52
#Mann= 3 , 0 , 0
       0     .03       0    5.59     .03       0   46.29     .03       0
Bank Sta=5.59,46.29
Exp/Cntr=0.5,0.3

Type RM Length L Ch R = 3 ,76.30   ,,,
BEGIN DESCRIPTION:
È­Á¤4±³(°³·®)
END DESCRIPTION:
Bridge Culvert--1,0,-1,-1, 0
Deck Dist Width WeirC Skew NumUp NumDn MinLoCord MaxHiCord MaxSubmerge Is_Ogee
0.1,19,1.44,0, 2, 2, , , 0.95, 0, 0,0,,
    5.59   46.29
      10      10
       9       9
    5.59   46.29
      10      10
       9       9
Pier Skew, UpSta & Num, DnSta & Num=  ,18.1, 2 ,18.1, 2 , 0 , 0 , 0 ,,
      .6      .6
     3.5       9
      .6      .6
     3.5       9
Pier Skew, UpSta & Num, DnSta & Num=  ,34.31, 2 ,34.31, 2 , 0 , 0 , 0 ,,
      .6      .6
     3.5       9
      .6      .6
     3.5       9
BR Coef=-1 , 0 , 0 ,, 0 ,,,0.8,-1,,0,
WSPro=,,,, 1 ,,,, 0 ,,,, 0 ,,,,-1 ,-1 ,-1 , 0 , 0 , 0 , 0 , 0
BC Design=,, 0 ,, 0 ,,,,,,

Type RM Length L Ch R = 1 ,76.20   ,20,20,20
#Sta/Elev= 19
       0    8.49    5.59    8.47    5.59    7.17    6.59    7.17    6.59    5.86
   10.59    4.46    11.1    4.28   23.33    4.28   25.73    3.08   31.83    3.08
   34.23    4.28   42.73    4.28   43.29    4.56   45.29    5.56   45.29    7.18
   46.29    7.18   46.29    8.48   49.99    8.48      60    8.52
#Mann= 3 , 0 , 0
       0     .03       0    5.59     .03       0   46.29     .03       0
Bank Sta=5.59,46.29
Exp/Cntr=0.5,0.3

Type RM Length L Ch R = 1 ,76      ,50,50,50
#Sta/Elev= 25
       0    8.01    5.29     7.8    5.79     7.8    5.79       8    8.79    8.23
    8.79    7.68    9.99    7.15   15.19    4.77    16.3    4.26   25.31    4.26
   27.71    3.06   31.71    3.06   35.31    4.26   43.29    4.26   43.29    5.06
   45.49    5.06   45.49    7.56   47.79    7.96   47.79    8.56   49.99    8.46
   51.59    8.46   51.59    8.26   52.09    8.26   58.69    8.33      60    8.35
#Mann= 3 , 0 , 0
       0     .03       0    8.79     .03       0   47.79     .03       0
Levee=-1,8.79,8.23,-1,47.79,8.56,,
Bank Sta=8.79,47.79
Exp/Cntr=0.3,0.1

Type RM Length L Ch R = 1 ,75      ,50,50,50
#Sta/Elev= 23
       0    7.77    5.28    7.59    5.68    7.59    7.38    7.52    7.38    7.72
    8.88    7.72   10.78    6.66   14.88    4.79   16.14    4.22   23.65    4.22
   26.05    3.02   30.05    3.02   33.65    4.22   41.51    4.22   42.48     4.7
   46.08    6.49   48.68    7.69   49.98    7.69   51.68    7.69   51.68    7.44
   52.18    7.44   58.48    7.64      60    7.59
#Mann= 3 , 0 , 0
       0     .03       0    8.88     .03       0   48.68     .03       0
Levee=-1,8.88,7.72,-1,48.68,7.69,,
Bank Sta=8.88,48.68
Exp/Cntr=0.3,0.1

Type RM Length L Ch R = 1 ,74      ,50,50,50
#Sta/Elev= 22
       0    7.68    5.28    7.56    5.78    7.56    7.28    7.61    8.68    7.81
   10.18    7.16   15.18    4.71   16.28    4.17   22.77    4.17   25.17    2.97
   29.17    2.97   32.77    4.17   41.31    4.17   42.18    4.56   46.18    6.36
   48.58    7.61   49.98    7.61   51.58    7.61   51.58    7.41   52.08    7.41
   58.58    7.61      60    7.58
#Mann= 3 , 0 , 0
       0     .03       0    8.68     .03       0   48.58     .03       0
Bank Sta=8.68,48.58
Exp/Cntr=0.3,0.1

Type RM Length L Ch R = 1 ,73      ,50,50,50
#Sta/Elev= 23
       0    7.48    5.58    7.39    6.08    7.39    7.58    7.32    7.58    7.52
    9.08    7.52   10.88    6.63   15.68     4.6   16.78    4.14   25.46    4.14
   27.86    2.94   31.86    2.94   35.46    4.14   41.78    4.14   42.98    4.74
   46.78    6.65   48.88    7.51   49.98    7.51   51.88    7.51   51.88    7.31
   52.38    7.31   58.78    7.47      60    7.46
#Mann= 3 , 0 , 0
       0     .03       0    9.08     .03       0   48.88     .03       0
Levee=-1,9.08,7.52,-1,48.88,7.51,,
Bank Sta=9.08,48.88
Exp/Cntr=0.3,0.1

Type RM Length L Ch R = 1 ,72      ,50,50,50
#Sta/Elev= 22
       0    7.44    5.48     7.3    5.98     7.3    7.58    7.27    9.08    7.47
   10.58    6.76   15.28     4.7    16.7    4.08   23.94    4.08   26.34    2.88
   30.34    2.88   33.94    4.08   41.49    4.08   42.68    4.63   46.88    6.58
   49.08    7.39   49.98    7.39   52.08    7.39   52.08    7.19   52.58    7.19
   58.88    7.44      60    7.43
#Mann= 3 , 0 , 0
       0     .03       0    9.08     .03       0   49.08     .03       0
Levee=-1,9.08,7.47,-1,49.08,7.39,,
Bank Sta=9.08,49.08
Exp/Cntr=0.3,0.1

Type RM Length L Ch R = 1 ,71      ,43,43,43
#Sta/Elev= 25
       0     7.6    5.68    7.45    6.18    7.45    6.18    7.65    9.18     7.8
    9.18    7.43   11.08    6.58   15.48    4.61   16.77    4.03   22.77    4.03
   25.17    2.83   29.17    2.83   32.77    4.03   41.97    4.03   42.98    4.51
   46.98    6.41   47.88    7.05   48.58    7.05   48.58     7.5   49.98     7.5
   51.88     7.5   51.88     7.3   52.38     7.3   58.98    7.55      60    7.53
#Mann= 3 , 0 , 0
       0     .03       0    9.18     .03       0   48.58     .03       0
Bank Sta=9.18,48.58
Exp/Cntr=0.3,0.1

Type RM Length L Ch R = 1 ,70.07   ,35,35,35
#Sta/Elev= 19
       0    8.07   11.48    8.07   11.48    7.27   12.48    7.27   12.48    5.81
   15.48    4.61   17.04    3.99   24.58    3.99   26.98    2.79   33.18    2.79
   35.58    3.99   42.57    3.99   43.48    4.51   45.98    5.95   45.98    7.27
   46.98    7.27   46.98    8.07   49.98    8.07      60    8.01
#Mann= 3 , 0 , 0
       0     .03       0   11.48     .03       0   46.98     .03       0
Levee=-1,11.48,8.07,-1,46.98,8.07,,
Bank Sta=11.48,46.98
Exp/Cntr=0.5,0.3

Type RM Length L Ch R = 3 ,69.3950 ,,,
BEGIN DESCRIPTION:
È­Á¤3±³
END DESCRIPTION:
Bridge Culvert--1,0,-1,-1, 0
Deck Dist Width WeirC Skew NumUp NumDn MinLoCord MaxHiCord MaxSubmerge Is_Ogee
0.1,34,1.44,0, 2, 2, , , 0.95, 0, 0,0,,
   11.48   46.98
    8.07    8.07
    7.27    7.27
   11.48   46.98
    8.07    8.07
    7.27    7.27
Pier Skew, UpSta & Num, DnSta & Num=  ,22.48, 2 ,22.48, 2 , 0 , 0 , 0 ,,
      .6      .6
     3.5       8
      .6      .6
     3.5       8
Pier Skew, UpSta & Num, DnSta & Num=  ,36.5, 2 ,36.5, 2 , 0 , 0 , 0 ,,
      .6      .6
     3.5       8
      .6      .6
     3.5       8
BR Coef=-1 , 0 , 0 ,, 0 ,,,0.8,-1,,0,
WSPro=,,,, 1 ,,,, 0 ,,,, 0 ,,,,-1 ,-1 ,-1 , 0 , 0 , 0 , 0 , 0
BC Design=,, 0 ,, 0 ,,,,,,

Type RM Length L Ch R = 1 ,69.22   ,22,22,22
#Sta/Elev= 19
       0    8.07   11.48    8.07   11.48    7.27   12.48    7.27   12.48    5.81
   15.48    4.61    17.1    3.96   24.65    3.96   27.05    2.76   33.25    2.76
   35.65    3.96   42.52    3.96   43.48    4.51   45.98    5.95   45.98    7.27
   46.98    7.27   46.98    8.07   49.98    8.07      60    8.01
#Mann= 3 , 0 , 0
       0     .03       0   11.48     .03       0   46.98     .03       0
Levee=-1,11.48,8.07,-1,46.98,8.07,,
Bank Sta=11.48,46.98
Exp/Cntr=0.5,0.3

Type RM Length L Ch R = 1 ,69      ,50,50,50
#Sta/Elev= 23
       0    7.63    5.68    7.57    6.18    7.57    6.18    7.77    9.18    7.77
    9.18    7.42   10.68    6.74   14.88    4.99   17.42    3.93   25.83    3.93
   28.23    2.73   32.23    2.73   35.83    3.93   45.98    3.93   45.98     4.1
   45.98     6.5   49.08    7.84   49.98    7.84   52.08    7.84   52.08    7.64
   52.58    7.64   58.98    7.76      60    7.75
#Mann= 3 , 0 , 0
       0     .03       0    9.18     .03       0   49.08     .03       0
Levee=-1,9.18,7.77,-1,49.08,7.84,,
Bank Sta=9.18,49.08
Exp/Cntr=0.3,0.1

Type RM Length L Ch R = 1 ,68      ,47,47,47
#Sta/Elev= 24
       0    7.17    5.78    6.97    6.28    6.97    7.68    7.04    7.68    7.24
    9.18    7.24   11.48    6.34   15.18     4.4   16.21    3.86   24.38    3.86
   26.78    2.66   30.78    2.66   34.38    3.86   41.58    3.86   43.08    4.51
   46.08    5.81   48.18    7.35   49.18    7.35   49.98    7.35   52.18    7.35
   52.18    7.15   52.68    7.15   59.18    7.28      60    7.26
#Mann= 3 , 0 , 0
       0     .03       0    9.18     .03       0   48.18     .03       0
Levee=-1,9.18,7.24,-1,48.18,7.35,,
Bank Sta=9.18,48.18
Exp/Cntr=0.3,0.1

Type RM Length L Ch R = 1 ,67.00   ,53,53,53
#Sta/Elev= 23
       0    7.32    6.38    7.12    6.88    7.12    8.38    7.47    8.38    7.32
    9.88    7.32   10.98     6.5   15.58    4.23   16.46    3.79   25.24    3.79
   27.64    2.59   31.64    2.59   35.24    3.79   41.81    3.79   43.28    4.46
   47.48    6.36   49.28    7.22   49.98    7.47   52.98    7.47   52.98    7.27
   53.48    7.27   59.58     7.4      60    7.39
#Mann= 3 , 0 , 0
       0     .03       0    9.88     .03       0   49.98     .03       0
Levee=-1,9.88,7.32,-1,49.98,7.47,,
Bank Sta=9.88,49.98
Exp/Cntr=0.5,0.3

Type RM Length L Ch R = 1 ,66      ,50,50,50
#Sta/Elev= 24
       0    7.04    6.08     6.9    6.58     6.9    8.08    6.96    8.08    7.16
    9.58    7.16   10.28    7.16   11.48    6.48   15.98     4.2   16.91    3.73
   25.55    3.73   27.95    2.53   31.95    2.53   35.55    3.73   42.09    3.73
   43.08    4.19   47.58     6.3   49.48    7.19   49.98    7.19   52.48    7.19
   52.48    6.99   52.98    6.99   59.58    7.19      60    7.18
#Mann= 3 , 0 , 0
       0     .03       0    9.58     .03       0   49.48     .03       0
Levee=-1,9.58,7.16,-1,49.48,7.19,,
Bank Sta=9.58,49.48
Exp/Cntr=0.3,0.1

Type RM Length L Ch R = 1 ,65      ,37,37,37
#Sta/Elev= 23
       0    7.19    6.28    7.03    6.68    7.03    6.68    7.23    9.48    7.26
   11.48    6.19   15.48    4.52   17.54    3.66   26.94    3.66   29.34    2.46
   33.34    2.46   36.94    3.66   42.12    3.66   42.88    4.04   47.18     6.2
   48.98    7.14   49.28    7.49   49.98    7.49   52.28    7.49   52.28    7.39
   52.78    7.39   59.38    7.53      60    7.52
#Mann= 3 , 0 , 0
       0     .03       0    9.48     .03       0   49.28     .03       0
Levee=-1,9.48,7.26,-1,49.28,7.49,,
Bank Sta=9.48,49.28
Exp/Cntr=0.3,0.1

Type RM Length L Ch R = 1 ,64.13   ,20,20,20
#Sta/Elev= 18
       0     7.9    9.98    7.84    9.98    7.04   10.98    7.04   10.98    6.22
   15.48    4.09   16.54    3.59   27.88    3.59   30.28    2.39   34.28    2.39
   37.88    3.59   44.56    3.59   45.48    4.02   48.98    5.66   48.98    7.03
   49.98    7.03   49.98    7.83      60    7.83
#Mann= 3 , 0 , 0
       0     .03       0    9.98     .03       0   49.98     .03       0
Levee=-1,9.98,7.84,-1,49.98,7.83,,
Bank Sta=9.98,49.98
Exp/Cntr=0.5,0.3

Type RM Length L Ch R = 3 ,64.03   ,,,
BEGIN DESCRIPTION:
È­Á¤2±³
END DESCRIPTION:
Bridge Culvert--1,0,-1,-1, 0
Deck Dist Width WeirC Skew NumUp NumDn MinLoCord MaxHiCord MaxSubmerge Is_Ogee
0.1,19,1.44,0, 2, 2, , , 0.95, 0, 0,0,,
    9.98   49.98
    7.84    7.84
    7.04    7.04
    9.98   49.98
    7.84    7.84
    7.04    7.04
Pier Skew, UpSta & Num, DnSta & Num=  ,22.48, 2 ,22.48, 2 , 0 , 0 , 0 ,,
      .6      .6
       3     8.7
      .6      .6
       3     8.7
Pier Skew, UpSta & Num, DnSta & Num=  ,39, 2 ,39, 2 , 0 , 0 , 0 ,,
      .6      .6
       3     8.7
      .6      .6
       3     8.7
BR Coef=-1 , 0 , 0 ,, 0 ,,,0.8,-1,,0,
WSPro=,,,, 1 ,,,, 0 ,,,, 0 ,,,,-1 ,-1 ,-1 , 0 , 0 , 0 , 0 , 0
BC Design=,, 0 ,, 0 ,,,,,,

Type RM Length L Ch R = 1 ,63.43   ,43,43,43
#Sta/Elev= 18
       0     7.9    9.98    7.84    9.98    7.04   10.98    7.04   10.98    6.22
   15.48    4.09   16.56    3.58   27.91    3.58   30.31    2.38   35.51    2.38
   37.91    3.58   41.77    3.58   45.48    4.65   48.98    5.66   48.98    7.03
   49.98    7.03   49.98    7.83      60    7.83
#Mann= 3 , 0 , 0
       0     .03       0    9.98     .03       0   49.98     .03       0
Levee=-1,9.98,7.84,-1,49.98,7.83,,
Bank Sta=9.98,49.98
Exp/Cntr=0.5,0.3

Type RM Length L Ch R = 1 ,63      ,50,50,50
#Sta/Elev= 22
       0    7.31    6.38    7.06    9.48    7.42    9.48    6.77   11.18    6.29
   15.78     3.9   16.46    3.55   23.71    3.55   26.11    2.35   30.11    2.35
   33.71    3.55   41.83    3.55   42.98    4.13   46.88    6.11   48.78     6.9
   48.78    7.35   49.98    7.35   51.68    7.35   51.68    7.15   52.18    7.15
   58.78     7.2      60    7.17
#Mann= 3 , 0 , 0
       0     .03       0    9.48     .03       0   48.78     .03       0
Levee=-1,9.48,7.42,-1,48.78,7.35,,
Bank Sta=9.48,48.78
Exp/Cntr=0.3,0.1

Type RM Length L Ch R = 1 ,62      ,50,50,50
#Sta/Elev= 22
       0    7.09    5.48    6.93    5.98    6.93    5.98    7.13    8.98    7.19
   10.68    6.33   15.28    4.01   16.28    3.51   28.36    3.51   30.76    2.31
   34.76    2.31   38.36    3.51   41.62    3.51   42.78    4.08   46.48    5.91
   48.68    7.12   49.98    7.12   51.68    7.12   51.68    6.92   52.18    6.92
   58.78    7.02      60    6.99
#Mann= 3 , 0 , 0
       0     .03       0    8.98     .03       0   48.68     .03       0
Bank Sta=8.98,48.68
Exp/Cntr=0.3,0.1

Type RM Length L Ch R = 1 ,61      ,50,50,50
#Sta/Elev= 22
       0    6.99    5.48    6.74    5.98    6.74    5.98    6.94    9.08    7.05
   11.08    5.92   14.98    4.18   16.58    3.47   25.71    3.47   28.11    2.27
   32.11    2.27   35.71    3.47   41.63    3.47   42.68    3.99   46.18    5.74
   48.98    7.09   49.98    7.09   51.98    7.09   51.98    6.89   52.48    6.89
   58.78    7.04      60    7.01
#Mann= 3 , 0 , 0
       0     .03       0    9.08     .03       0   48.98     .03       0
Levee=-1,9.08,7.05,-1,48.98,7.09,,
Bank Sta=9.08,48.98
Exp/Cntr=0.3,0.1

Type RM Length L Ch R = 1 ,60      ,50,50,50
#Sta/Elev= 22
       0    6.92     5.9     6.7     6.4     6.7     6.4     6.9     9.5    7.05
    11.1    6.15    15.9       4   17.18    3.43   28.01    3.43   30.41    2.23
   34.41    2.23   38.01    3.43   42.03    3.43    42.9    3.85    46.4    5.55
    49.3    7.05    50.1    7.05    52.3    7.05    52.3    6.85    52.7    6.85
    59.4       7      60    6.98
#Mann= 3 , 0 , 0
       0     .03       0     9.5     .03       0    49.3     .03       0
Levee=-1,9.5,7.05,-1,49.3,7.05,,
Bank Sta=9.5,49.3
Exp/Cntr=0.3,0.1

Type RM Length L Ch R = 1 ,59      ,50,50,50
#Sta/Elev= 22
       0    6.81     6.1    6.61     6.6    6.61     6.6    6.81     9.5    6.91
    11.4    5.93    15.9    3.95   17.18    3.39   30.06    3.39   32.46    2.19
   36.46    2.19   40.06    3.39   42.47    3.39    43.4    3.84    47.8    5.98
    49.3    6.86    50.1    6.86    52.3    6.76    52.3    6.56    52.8    6.56
    59.4    6.71      60    6.71
#Mann= 3 , 0 , 0
       0     .03       0     9.5     .03       0    49.3     .03       0
Levee=-1,9.5,6.91,-1,49.3,6.86,,
Bank Sta=9.5,49.3
Exp/Cntr=0.3,0.1

Type RM Length L Ch R = 1 ,58      ,50,50,50
#Sta/Elev= 22
       0    6.69     6.1    6.47     6.6    6.47     6.6    6.67     9.6    6.78
    11.5    5.71    15.3    3.98   16.69    3.35    30.1    3.35    32.5    2.15
    36.5    2.15    40.1    3.35   42.44    3.35    43.5    3.81      47    5.34
    49.3     6.8    50.1     6.8    52.3     6.8    52.3    6.55    52.8    6.55
    59.4     6.6      60     6.6
#Mann= 3 , 0 , 0
       0     .03       0     9.6     .03       0    49.3     .03       0
Levee=-1,9.6,6.78,-1,49.3,6.8,,
Bank Sta=9.6,49.3
Exp/Cntr=0.3,0.1

Type RM Length L Ch R = 1 ,57      ,50,50,50
#Sta/Elev= 22
       0    6.58     6.1    6.39     6.6    6.39     6.6    6.59     9.6    6.68
    10.8    6.09      15    4.08   16.61    3.31   30.18    3.31   32.58    2.11
   36.58    2.11   40.18    3.31   42.38    3.31    43.4    3.77      47     5.4
    49.3    6.72    50.1    6.72    52.3    6.72    52.3    6.52    52.8    6.52
    59.2    6.61      60     6.6
#Mann= 3 , 0 , 0
       0     .03       0     9.6     .03       0    49.3     .03       0
Levee=-1,9.6,6.68,-1,49.3,6.72,,
Bank Sta=9.6,49.3
Exp/Cntr=0.3,0.1

Type RM Length L Ch R = 1 ,56      ,50,50,50
#Sta/Elev= 22
       0    6.63     6.3     6.4     6.8     6.4     6.8     6.6     9.8     6.7
    11.5     5.8    15.9    3.85   17.23    3.26   30.46    3.26   32.86    2.06
   36.86    2.06   40.46    3.26   42.79    3.26    43.9     3.8    47.8    5.69
    49.6    6.68    50.1    6.68    52.6    6.63    52.6    6.43    53.1    6.43
    59.6    6.58      60    6.58
#Mann= 3 , 0 , 0
       0     .03       0     9.8     .03       0    49.6     .03       0
Levee=-1,9.8,6.7,-1,49.6,6.68,,
Bank Sta=9.8,49.6
Exp/Cntr=0.3,0.1

Type RM Length L Ch R = 1 ,55      ,50,50,50
#Sta/Elev= 22
       0    6.49     6.4     6.3     6.9     6.3     6.9     6.5     9.9    6.56
    11.7    5.53    15.3    3.94   16.91    3.23   30.46    3.23   32.86    2.03
   36.86    2.03   40.46    3.23   42.88    3.23    43.8    3.69    47.7    5.65
    49.6    6.65    50.1    6.65    52.6     6.6    52.6     6.4    53.1     6.4
    59.6    6.61      60     6.6
#Mann= 3 , 0 , 0
       0     .03       0     9.9     .03       0    49.6     .03       0
Levee=-1,9.9,6.56,-1,49.6,6.65,,
Bank Sta=9.9,49.6
Exp/Cntr=0.3,0.1

Type RM Length L Ch R = 1 ,54      ,50,50,50
#Sta/Elev= 22
       0    6.59     6.4    6.28     6.9    6.28     6.9    6.48     9.8    6.64
    11.3    5.72    14.9    4.07   16.82    3.19   27.51    3.19   29.91    1.99
   33.91    1.99   37.51    3.19   42.75    3.19    44.1    3.83    47.8    5.58
    49.6    6.61    50.1    6.61    52.6    6.51    52.6    6.31    53.1    6.31
    59.6    6.56      60    6.55
#Mann= 3 , 0 , 0
       0     .03       0     9.8     .03       0    49.6     .03       0
Levee=-1,9.8,6.64,-1,49.6,6.61,,
Bank Sta=9.8,49.6
Exp/Cntr=0.3,0.1

Type RM Length L Ch R = 1 ,53      ,2.1,2.1,2.1
#Sta/Elev= 24
       0    6.48      .1    6.48     6.6    6.59     7.1    6.59     7.1    6.79
      10    6.79      10    6.95    10.2    6.95    10.2    6.34    11.8    3.75
   12.17    3.15   25.18    3.15   27.58    1.95   31.58    1.95   35.18    3.15
    49.6    3.15    49.6     3.9    49.6    6.85    50.1    6.85    52.6    6.85
    52.6    6.65    53.1    6.65    59.5    6.72      60    6.71
#Mann= 3 , 0 , 0
       0     .03       0      10     .03       0    49.6     .03       0
Levee=-1,10,6.79,-1,49.6,6.85,,
Bank Sta=10,49.6
Exp/Cntr=0.3,0.1

Type RM Length L Ch R = 1 ,52.479  ,20.9,20.9,20.9
#Sta/Elev= 18
       0    6.59     9.6    6.83     9.6    5.33    10.6    5.33    10.6    3.85
    10.6    3.13   26.05    3.13   28.45    1.93   33.65    1.93   36.05    3.13
    48.6    3.13    48.6    3.45    48.6    5.28    49.6    5.28    49.6    6.78
    50.1    6.78    59.5    6.33      60    6.33
#Mann= 3 , 0 , 0
       0     .03       0     9.6     .03       0    49.6     .03       0
Levee=-1,9.6,6.83,-1,49.6,6.78,,
Bank Sta=9.6,49.6
Exp/Cntr=0.5,0.3

Type RM Length L Ch R = 3 ,52.3745 ,,,
BEGIN DESCRIPTION:
È­¶û±³(°³·®)
END DESCRIPTION:
Bridge Culvert--1,0,-1,-1, 0
Deck Dist Width WeirC Skew NumUp NumDn MinLoCord MaxHiCord MaxSubmerge Is_Ogee
0.1,20,1.44,0, 2, 2, , , 0.95, 0, 0,0,,
     9.6    49.6
       9       9
     8.5     8.5
     9.6    49.6
       9       9
     8.5     8.5
Pier Skew, UpSta & Num, DnSta & Num=  ,22.1, 2 ,22.1, 2 , 0 , 0 , 0 ,,
      .7      .7
       2       7
      .7      .7
       2       7
Pier Skew, UpSta & Num, DnSta & Num=  ,37, 2 ,37, 2 , 0 , 0 , 0 ,,
      .7      .7
       2       7
      .7      .7
       2       7
BR Coef=-1 , 0 , 0 ,, 0 ,,,0.8,-1,,0,
WSPro=,,,, 1 ,,,, 0 ,,,, 0 ,,,,-1 ,-1 ,-1 , 0 , 0 , 0 , 0 , 0
BC Design=,, 0 ,, 0 ,,,,,,

Type RM Length L Ch R = 1 ,52.27   ,27,27,27
#Sta/Elev= 18
       0    6.59     9.6    6.83     9.6    5.33    10.6    5.33    10.6    3.85
    10.6    3.13   26.05    3.13   28.45    1.93   33.65    1.93   36.05    3.13
    48.6    3.13    48.6    3.45    48.6    5.28    49.6    5.28    49.6    6.78
    50.1    6.78    59.5    6.33      60    6.33
#Mann= 3 , 0 , 0
       0     .03       0     9.6     .03       0    49.6     .03       0
Levee=-1,9.6,6.83,-1,49.6,6.78,,
Bank Sta=9.6,49.6
Exp/Cntr=0.5,0.3

Type RM Length L Ch R = 1 ,52      ,50,50,50
#Sta/Elev= 23
       0    6.43      .1    6.43     6.6    6.25     7.1    6.25     7.1    6.45
    10.1    6.47      12    5.53    14.9    4.07   16.81    3.11    26.1    3.11
    28.5    1.91    32.5    1.91    36.1    3.11   42.92    3.11    44.1    3.67
    47.8    5.42    49.9    6.47    50.1    6.47    52.9    6.47    52.9    6.27
    53.4    6.27    59.8    6.44      60    6.43
#Mann= 3 , 0 , 0
       0     .03       0    10.1     .03       0    49.9     .03       0
Levee=-1,10.1,6.47,-1,49.9,6.47,,
Bank Sta=10.1,49.9
Exp/Cntr=0.3,0.1

Type RM Length L Ch R = 1 ,51      ,50,50,50
#Sta/Elev= 23
       0    6.37      .1    6.37     6.6    6.12     7.1    6.12     7.1    6.32
    10.1     6.4    11.9    5.59    15.5       4   17.61    3.07   27.56    3.07
   29.96    1.87   33.96    1.87   37.56    3.07    43.3    3.07    44.2    3.54
    47.4     5.2    49.9    6.45    50.1    6.45    52.9    6.35    52.9    6.15
    53.4    6.15    59.9    6.28      60    6.28
#Mann= 3 , 0 , 0
       0     .03       0    10.1     .03       0    49.9     .03       0
Levee=-1,10.1,6.4,-1,49.9,6.45,,
Bank Sta=10.1,49.9
Exp/Cntr=0.3,0.1

Type RM Length L Ch R = 1 ,50      ,50,50,50
#Sta/Elev= 22
       0    6.27      .3    6.28     6.7    6.03     7.2    6.03     7.2    6.23
    10.1    6.39      12    5.52    15.8    3.64   17.01    3.04   30.02    3.04
   32.42    1.84   36.42    1.84   40.02    3.04   43.13    3.04    44.1    3.51
      48    5.39    49.9    6.37    50.1    6.37    52.9    6.27    52.9    6.07
    53.4    6.07      60     6.3
#Mann= 3 , 0 , 0
       0     .03       0    10.1     .03       0    49.9     .03       0
Levee=-1,10.1,6.39,-1,49.9,6.37,,
Bank Sta=10.1,49.9
Exp/Cntr=0.3,0.1
