HEC-RAS study hj.prj: Hwajung_plan

--- hj.g01 (geometry) --- (continued)

Type RM Length L Ch R = 1 ,49      ,50,50,50
#Sta/Elev= 22
       0    6.36      .4    6.38     6.8    6.17     7.3    6.17     7.3    6.37
    10.3    6.45    12.1    5.54    15.8     3.7   17.18    3.01   28.54    3.01
   30.94    1.81   34.94    1.81   38.54    3.01   43.05    3.01    44.3    3.62
    47.9    5.36      50    6.35    50.1    6.35      53    6.33      53    6.13
    53.6    6.13      60    6.32
#Mann= 3 , 0 , 0
       0     .03       0    10.3     .03       0      50     .03       0
Levee=-1,10.3,6.45,-1,50,6.35,,
Bank Sta=10.3,50
Exp/Cntr=0.3,0.1

Type RM Length L Ch R = 1 ,48      ,50,50,50
#Sta/Elev= 22
       0    6.33      .2    6.34     6.7    6.13     7.2    6.13     7.2    6.33
    10.2    6.34      12     5.5    15.7    3.71    17.2    2.99   30.95    2.99
   33.35    1.79   37.35    1.79   40.95    2.99   42.85    2.99    44.2    3.57
    47.2    4.87      50    6.36    50.2    6.36      53    6.36      53    6.16
    53.5    6.16      60     6.2
#Mann= 3 , 0 , 0
       0     .03       0    10.2     .03       0      50     .03       0
Levee=-1,10.2,6.34,-1,50,6.36,,
Bank Sta=10.2,50
Exp/Cntr=0.3,0.1

Type RM Length L Ch R = 1 ,47      ,50,50,50
#Sta/Elev= 23
       0    6.23    6.65    5.97    7.25    5.97    7.25    6.17   10.25    6.28
   12.05    5.44   15.55    3.71   17.07    2.96   31.05    2.96   33.45    1.76
   37.45    1.76   41.05    2.96   43.15    2.96   44.75    3.71   48.55    5.49
   49.75    6.18   49.95    6.26   50.45    6.26   52.95    6.26   52.95    6.06
   53.45    6.06   59.95     6.1      60     6.1
#Mann= 3 , 0 , 0
       0     .03       0   10.25     .03       0   49.95     .03       0
Levee=-1,10.25,6.28,-1,49.95,6.26,,
Bank Sta=10.25,49.95
Exp/Cntr=0.3,0.1

Type RM Length L Ch R = 1 ,46      ,50,50,50
#Sta/Elev= 22
       0       6      .4    6.02     6.6    5.84     7.2    5.84     7.2    6.04
    10.1    6.12      12     5.2    15.3    3.61   16.71    2.93   31.24    2.93
   33.64    1.73   37.64    1.73   41.24    2.93   43.29    2.93    44.3    3.43
    48.1     5.3      50    6.16    50.2    6.16      53    6.06      53    5.86
    53.5    5.86      60    6.01
#Mann= 3 , 0 , 0
       0     .03       0    10.1     .03       0      50     .03       0
Levee=-1,10.1,6.12,-1,50,6.16,,
Bank Sta=10.1,50
Exp/Cntr=0.3,0.1

Type RM Length L Ch R = 1 ,45      ,50,50,50
#Sta/Elev= 21
       0    6.05       1    6.09     7.6    5.87     8.2    5.87    11.2    6.12
      13    5.07    15.9    3.63   17.37     2.9   31.46     2.9   33.86     1.7
   37.86     1.7   41.46     2.9   44.01     2.9    45.3    3.46    49.3    5.19
    50.8    5.96    52.5    5.96    53.8    5.96    53.8    5.76    54.3    5.76
      60    5.85
#Mann= 3 , 0 , 0
       0     .03       0    11.2     .03       0    50.8     .03       0
Levee=-1,11.2,6.12,-1,50.8,5.96,,
Bank Sta=11.2,50.8
Exp/Cntr=0.3,0.1

Type RM Length L Ch R = 1 ,44      ,50,50,50
#Sta/Elev= 24
       0    6.14     2.2    6.23     8.7    5.99     9.3    5.99     9.3    6.19
    12.4    6.23    12.4    5.83      14    5.12    21.1     3.6   24.49    2.87
   33.85    2.87   36.25    1.67   40.25    1.67   43.85    2.87   45.57    2.87
    46.8    3.43    50.9    5.29    52.4     5.7    52.4       6    52.5       6
    55.4     5.9    55.4     5.7    55.9     5.7      60     5.9
#Mann= 3 , 0 , 0
       0     .03       0    12.4     .03       0    52.4     .03       0
Levee=-1,12.4,6.23,-1,52.4,7,,
Bank Sta=12.4,52.4
Exp/Cntr=0.3,0.1

Type RM Length L Ch R = 1 ,43      ,50,50,50
#Sta/Elev= 24
       0     6.3     2.2    6.39     8.6    6.16     9.2    6.16     9.2    6.41
    12.2    6.37    12.2    5.97    13.7    5.27    17.1    3.48    18.3    2.85
   32.85    2.85   35.25    1.65   39.25    1.65   42.85    2.85   45.23    2.85
    46.3    3.33    51.1    5.51      52    5.97      52    6.42    52.5    6.42
      55    6.32      55    6.12    55.5    6.12      60    6.19
#Mann= 3 , 0 , 0
       0     .03       0    12.2     .03       0      52     .03       0
Bank Sta=12.2,52
Exp/Cntr=0.3,0.1

Type RM Length L Ch R = 1 ,42      ,4.7,4.7,4.7
#Sta/Elev= 19
       0    6.79   12.95    6.73   12.95    6.17   13.75    6.17   13.75    4.67
   16.25    3.69   18.47    2.82   28.18    2.82   30.58    1.62   36.43    1.62
   38.83    2.82   45.46    2.82   47.25    3.41   50.45    4.47   50.45    6.12
   51.25    6.12   51.25    6.77   54.25    6.72      60     6.7
#Mann= 3 , 0 , 0
       0     .03       0   12.95     .03       0   51.25     .03       0
Bank Sta=12.95,51.25
Exp/Cntr=0.3,0.1

Type RM Length L Ch R = 1 ,41.453  ,43.3,43.3,43.3
#Sta/Elev= 19
       0     6.8   14.45    6.73   14.45    6.17   15.25    6.17   15.25    4.67
   17.75    3.69   20.05    2.79   29.75    2.79   32.15    1.59   37.85    1.59
   40.25    2.79   46.88    2.79   48.75    3.41   51.95    4.47   51.95    6.12
   52.75    6.12   52.75    6.77   55.75    6.72      60     6.7
#Mann= 3 , 0 , 0
       0     .03       0   14.45     .03       0   52.75     .03       0
Bank Sta=14.45,52.75
Exp/Cntr=0.5,0.3

Type RM Length L Ch R = 3 ,41.2365 ,,,
BEGIN DESCRIPTION:
È­Á¤1±³
END DESCRIPTION:
Bridge Culvert--1,0,-1,-1, 0
Deck Dist Width WeirC Skew NumUp NumDn MinLoCord MaxHiCord MaxSubmerge Is_Ogee
0.1,43,1.44,0, 2, 2, , , 0.95, 0, 0,0,,
   14.45   52.75
    6.73    6.73
    6.17    6.17
   14.45   52.75
    6.73    6.73
    6.17    6.17
Pier Skew, UpSta & Num, DnSta & Num=  ,22.75, 2 ,22.75, 2 , 0 , 0 , 0 ,,
       1       1
       2       7
       1       1
       2       7
Pier Skew, UpSta & Num, DnSta & Num=  ,40.75, 2 ,40.75, 2 , 0 , 0 , 0 ,,
       1       1
       2       7
       1       1
       2       7
BR Coef=-1 , 0 , 0 ,, 0 ,,,0.8,-1,,0,
WSPro=,,,, 1 ,,,, 0 ,,,, 0 ,,,,-1 ,-1 ,-1 , 0 , 0 , 0 , 0 , 0
BC Design=,, 0 ,, 0 ,,,,,,

Type RM Length L Ch R = 1 ,41.02   ,2,2,2
#Sta/Elev= 19
       0     6.8   14.45    6.73   14.45    6.17   15.25    6.17   15.25    4.67
   17.75    3.69   20.05    2.79   29.75    2.79   32.15    1.59   37.85    1.59
   40.25    2.79   46.88    2.79   48.75    3.41   51.95    4.47   51.95    6.12
   52.75    6.12   52.75    6.77   55.75    6.72      60     6.7
#Mann= 3 , 0 , 0
       0     .03       0   14.45     .03       0   52.75     .03       0
Bank Sta=14.45,52.75
Exp/Cntr=0.5,0.3

Type RM Length L Ch R = 1 ,41      ,50,50,50
#Sta/Elev= 24
       0    6.65    2.35    6.66    8.85    6.48    9.35    6.48   13.05    6.81
   13.05    5.81   14.35    4.91   17.65    3.24   18.54    2.79   28.91    2.79
   31.31    1.59   35.31    1.59   38.91    2.79   46.77    2.79   47.05    2.93
   50.15    4.49   52.15    5.55   52.35    5.55   52.35    6.15   52.85    6.15
   55.35    6.05   55.35    5.85   55.85    5.85      60    5.94
#Mann= 3 , 0 , 0
       0     .03       0   13.05     .03       0   52.35     .03       0
Bank Sta=13.05,52.35
Exp/Cntr=0.3,0.1

Type RM Length L Ch R = 1 ,40      ,50,50,50
#Sta/Elev= 22
       0    6.07    3.05    6.13    9.55    5.91   10.05    5.91   10.05    6.06
   12.95    6.13   18.35    3.28   19.57    2.64   26.78    2.64   29.18    1.44
   33.18    1.44   36.78    2.64   43.22    2.64   45.15    3.46   47.15    3.46
   50.35    4.85   52.25    5.93   52.75    5.98   55.75    5.88   55.75    5.68
   56.25    5.68      60    5.78
#Mann= 3 , 0 , 0
       0     .03       0   12.95     .03       0   52.75     .03       0
Levee=-1,12.95,6.13,-1,52.75,5.98,,
Bank Sta=12.95,52.75
Exp/Cntr=0.3,0.1

Type RM Length L Ch R = 1 ,39      ,50,50,50
#Sta/Elev= 23
       0    5.71     3.2    5.78     9.5    5.57      10    5.57      10    5.77
    13.2    5.86    14.8    4.92      18    3.18   19.28    2.49   33.11    2.49
   35.51    1.29   39.51    1.29   43.11    2.49   45.43    2.49      47    3.25
    50.6       5    52.1    5.67    52.7    5.77    52.9    5.77    55.7    5.67
    55.7    5.47    56.2    5.47      60    5.55
#Mann= 3 , 0 , 0
       0     .03       0    13.2     .03       0    52.7     .03       0
Levee=-1,13.2,5.86,-1,52.7,5.77,,
Bank Sta=13.2,52.7
Exp/Cntr=0.3,0.1

Type RM Length L Ch R = 1 ,38      ,50,50,50
#Sta/Elev= 22
       0    5.82     1.9    5.86     8.3    5.61     8.8    5.61     8.8    5.81
      12    5.91      14    5.08    17.4    3.26   19.13    2.33    28.6    2.33
      31    1.13      35    1.13    38.6    2.33   46.22    2.33    49.5    4.72
      51    5.81      52    5.81    52.5    5.81      55    5.71      55    5.51
    55.5    5.51      60    5.58
#Mann= 3 , 0 , 0
       0     .03       0      12     .03       0      51     .03       0
Levee=-1,12,5.91,-1,51,5.81,,
Bank Sta=12,51
Exp/Cntr=0.3,0.1

Type RM Length L Ch R = 1 ,37      ,50,50,50
#Sta/Elev= 22
       0     5.7     1.7    5.73     8.2    5.56     8.7    5.56     8.7    5.76
    11.7    5.91    13.3    5.04    16.5    3.36   18.75    2.18   29.36    2.18
   31.76     .98   35.76     .98   39.36    2.18    43.6    2.18    45.4    3.03
    48.9    4.68    51.1    5.71    52.5    5.71    54.1    5.61    54.1    5.41
    54.6    5.41      60    5.51
#Mann= 3 , 0 , 0
       0     .03       0    11.7     .03       0    51.1     .03       0
Bank Sta=11.7,51.1
Exp/Cntr=0.3,0.1

Type RM Length L Ch R = 1 ,36      ,50,50,50
#Sta/Elev= 23
       0     5.6     2.5    5.65     8.8    5.38     9.3    5.38     9.3    5.58
    12.5    5.71    13.2    5.55    14.2    4.89    17.1    3.36   19.63    2.03
   24.35    2.03   26.75     .83   39.95     .83   42.35    2.03   44.68    2.03
    46.3    2.85    50.1    4.78    51.9    5.65    52.5    5.65    54.9    5.55
    54.9    5.35    55.4    5.35      60    5.43
#Mann= 3 , 0 , 0
       0     .03       0    12.5     .03       0    51.9     .03       0
Bank Sta=12.5,51.9
Exp/Cntr=0.3,0.1

Type RM Length L Ch R = 1 ,35      ,50,50,50
#Sta/Elev= 21
       0    5.43     2.7    5.49     9.1    5.36     9.6    5.36     9.6    5.56
    12.8    5.59    14.5    4.69    18.5       3   21.16    1.88   27.55    1.88
   29.95     .68   33.95     .68   37.55    1.88   44.43    1.88    46.7    3.01
      52    5.66    52.5    5.66      55    5.56      55    5.36    55.5    5.36
      60    5.52
#Mann= 3 , 0 , 0
       0     .03       0    12.8     .03       0      52     .03       0
Bank Sta=12.8,52
Exp/Cntr=0.3,0.1

Type RM Length L Ch R = 1 ,34      ,50,50,50
#Sta/Elev= 21
       0    5.61     6.1    5.43     6.6    5.43     6.6    5.58     9.8    5.71
    11.4    4.95    15.1    3.08   17.78    1.72   22.07    1.72   24.47     .52
   28.47     .52   32.07    1.72   41.18    1.72    44.1    3.04    47.6    4.62
    49.5    5.62    52.5    5.57    52.5    5.37      53    5.37    59.7    5.62
      60    5.61
#Mann= 3 , 0 , 0
       0     .03       0     9.8     .03       0    49.5     .03       0
Bank Sta=9.8,49.5
Exp/Cntr=0.3,0.1

Type RM Length L Ch R = 1 ,33      ,42,42,42
#Sta/Elev= 21
       0     5.7     3.2    5.73     9.6    5.53    10.1    5.53    10.1    5.73
    13.2    5.85      15    4.75    18.5    2.88   20.95    1.57    26.7    1.57
    29.1     .37    35.1     .37    38.7    1.57   44.73    1.57    47.6    3.12
    52.5    5.76      54    5.74    55.5    5.69    55.5    5.49      56    5.49
      60    5.64
#Mann= 3 , 0 , 0
       0     .03       0    13.2     .03       0    52.5     .03       0
Bank Sta=13.2,52.5
Exp/Cntr=0.3,0.1

Type RM Length L Ch R = 1 ,32.08   ,70,70,70
#Sta/Elev= 21
       0    6.77     6.3    6.67     6.8    6.67    10.5    6.75    10.5    6.15
    11.1    6.15    11.1    4.77   16.39    1.42   23.31    1.42   25.71     .22
   32.91     .22   35.31    1.42   41.95    1.42      42    1.46    44.9     3.8
    44.9    6.05    45.5    6.05    45.5    6.65      55    6.51    58.7    6.45
      60    6.41
#Mann= 3 , 0 , 0
       0     .03       0    10.5     .03       0    45.5     .03       0
Bank Sta=10.5,45.5
Exp/Cntr=0.3,0.1

Type RM Length L Ch R = 3 ,31.23   ,,,
BEGIN DESCRIPTION:
È­Á¤±³
END DESCRIPTION:
Bridge Culvert--1,0,-1,-1, 0
Deck Dist Width WeirC Skew NumUp NumDn MinLoCord MaxHiCord MaxSubmerge Is_Ogee
0.1,69,1.44,0, 2, 2, , , 0.95, 0, 0,0,,
    10.5    45.5
    6.75    6.65
    6.15    6.05
    10.5    45.5
    6.58    6.58
    5.98    5.98
Pier Skew, UpSta & Num, DnSta & Num=  ,21, 2 ,21, 2 , 0 , 0 , 0 ,,
      .6      .6
       0       7
      .6      .6
       0       7
Pier Skew, UpSta & Num, DnSta & Num=  ,34.5, 2 ,34.5, 2 , 0 , 0 , 0 ,,
      .6      .6
       0       7
      .6      .6
       0       7
BR Coef=-1 , 0 , 0 ,, 0 ,,,0.8,-1,,0,
WSPro=,,,, 1 ,,,, 0 ,,,, 0 ,,,,-1 ,-1 ,-1 , 0 , 0 , 0 , 0 , 0
BC Design=,, 0 ,, 0 ,,,,,,

Type RM Length L Ch R = 1 ,30.38   ,24,24,24
#Sta/Elev= 18
       0    6.64    10.5    6.58    10.5    5.98    11.1    5.98    11.1    4.69
   16.38    1.36    23.3    1.36    25.7     .16    32.9     .16    35.3    1.36
   41.96    1.36      42    1.39    44.9    3.73    44.9    5.98    45.5    5.98
    45.5    6.58      55    6.57      60    6.55
#Mann= 3 , 0 , 0
       0     .03       0    10.5     .03       0    45.5     .03       0
Bank Sta=10.5,45.5
Exp/Cntr=0.5,0.3

Type RM Length L Ch R = 1 ,30.14   ,11,11,11
#Sta/Elev= 26
       0    7.38       0    7.36    16.6    6.86    18.1    6.58    19.3    7.27
    23.6       7    32.4    7.16    40.1    6.75    42.4    5.39    47.6    5.39
    50.3    3.66    52.5    2.65    53.9       2   57.82     .92   63.03     .92
   64.63     .12   71.43     .12   73.03     .92   82.61     .92    88.4    3.78
    94.6    6.55    95.6    6.55   101.6    6.55   102.9    6.41   128.1    6.48
   152.8    6.48
#Mann= 3 , 0 , 0
       0     .03       0    47.6     .03       0    94.6     .03       0
Bank Sta=47.6,94.6
Exp/Cntr=0.5,0.3

Type RM Length L Ch R = 3 ,30.085  ,,,
BEGIN DESCRIPTION:
ÁöÇÏÃ¶±³·®
END DESCRIPTION:
Bridge Culvert--1,0,-1,-1, 0
Deck Dist Width WeirC Skew NumUp NumDn MinLoCord MaxHiCord MaxSubmerge Is_Ogee
0.1,10,1.44,0, 2, 2, , , 0.95, 0, 0,0,,
       0     153
      10      10
      10      10
       0     153
      10      10
      10      10
Pier Skew, UpSta & Num, DnSta & Num=  ,54, 2 ,54, 2 , 0 , 0 , 0 ,,
     1.5     1.5
       0      10
     1.5     1.5
       0      10
Pier Skew, UpSta & Num, DnSta & Num=  ,78.6, 2 ,78.6, 2 , 0 , 0 , 0 ,,
     1.5     1.5
       0      10
     1.5     1.5
       0      10
BR Coef=-1 , 0 , 0 ,, 0 ,,,0.8,-1,,0,
WSPro=,,,, 1 ,,,, 0 ,,,, 0 ,,,,-1 ,-1 ,-1 , 0 , 0 , 0 , 0 , 0
BC Design=,, 0 ,, 0 ,,,,,,

Type RM Length L Ch R = 1 ,30.03   ,3,3,3
#Sta/Elev= 26
       0    7.38       0    7.36    16.6    6.86    18.1    6.58    19.3    7.27
    23.6       7    32.4    7.16    40.1    6.75    42.4    5.39    47.6    5.39
    50.3    3.66    52.5    2.65    53.9       2   57.82     .92   63.03     .92
   64.63     .12   71.43     .12   73.03     .92   82.61     .92    88.4    3.78
    94.6    6.55    95.6    6.55   101.6    6.55   102.9    6.41   128.1    6.48
   152.8    6.48
#Mann= 3 , 0 , 0
       0     .03       0    47.6     .03       0    94.6     .03       0
Bank Sta=47.6,94.6
Exp/Cntr=0.5,0.3

Type RM Length L Ch R = 1 ,30      ,50,50,50
#Sta/Elev= 17
       0    6.61    32.8    5.31    38.1     5.2    40.8    3.67   46.86     .92
   51.96     .92   53.56     .12   60.36     .12   61.96     .92   73.42     .92
    79.2    3.77      85    6.33    86.3    6.33    88.1    6.48    90.1    6.48
   126.8    6.08   156.8    6.08
#Mann= 3 , 0 , 0
       0     .03       0    38.1     .03       0      85     .03       0
Bank Sta=38.1,85
Exp/Cntr=0.3,0.1

Type RM Length L Ch R = 1 ,29      ,50,50,50
#Sta/Elev= 29
       0    5.62      30    5.77    32.5    5.77    42.5    5.95    51.4    8.07
    58.5    8.07      68    5.41    73.5    5.29    76.2     3.7    82.3     .87
   89.05     .87   90.65     .07   97.45     .07   99.05     .87  113.04     .87
   119.1    3.61   122.5    5.07     124    5.07   125.5    5.17   127.5    5.17
   130.4    5.17   130.7    4.86   131.4    4.86   132.5     5.5   136.5     5.5
   145.2    5.62   150.5    7.17   164.9    9.24     185    9.64
#Mann= 3 , 0 , 0
       0     .03       0    73.5     .03       0   122.5     .03       0
Bank Sta=73.5,122.5
Exp/Cntr=0.3,0.1

Type RM Length L Ch R = 1 ,28      ,12,12,12
#Sta/Elev= 22
       0    4.97      30    5.17    32.5    5.17    43.3    5.29    71.3    5.22
    73.8    3.82   79.79     .81   91.67     .81   93.27     .01  100.07     .01
  101.67     .81  114.78     .81   120.9    3.67   123.8    5.17     125    5.17
     127    5.17   129.4    5.17   130.1    4.71   130.7    4.71   131.3     5.1
   135.3     5.1   158.6    6.01
#Mann= 3 , 0 , 0
       0     .03       0    71.3     .03       0   123.8     .03       0
Bank Sta=71.3,123.8
Exp/Cntr=0.3,0.1

Type RM Length L Ch R = 1 ,27.38   ,30,30,30
#Sta/Elev= 23
       0    4.72    25.7    4.91    35.7    4.82      54    4.97      54       4
   54.85       4   54.85    3.63      56    3.63   61.96     .77   74.86     .77
   76.46    -.03   83.26    -.03   84.86     .77   97.23     .77     102    3.63
  103.15    3.63  103.15       4     104       4     104    4.99   125.8    4.94
   133.8    5.02   142.1    4.91     161     4.7
#Mann= 3 , 0 , 0
       0     .03       0      54     .03       0     104     .03       0
Bank Sta=54,104
Exp/Cntr=0.5,0.3

Type RM Length L Ch R = 3 ,27.23   ,,,
BEGIN DESCRIPTION:
È­Á¤11±³(È¾´Ü¼öÁ¤)
END DESCRIPTION:
Bridge Culvert--1,0,-1,-1, 0
Deck Dist Width WeirC Skew NumUp NumDn MinLoCord MaxHiCord MaxSubmerge Is_Ogee
0.1,29,1.44,0, 2, 2, , , 0.95, 0, 0,0,,
      54     104
    4.97    4.99
       4       4
      54     104
    4.97    4.99
       4       4
Pier Skew, UpSta & Num, DnSta & Num=  ,71, 2 ,71, 2 , 0 , 0 , 0 ,,
       1       1
       0       5
       1       1
       0       5
Pier Skew, UpSta & Num, DnSta & Num=  ,88, 2 ,88, 2 , 0 , 0 , 0 ,,
       1       1
       0       5
       1       1
       0       5
BR Coef=-1 , 0 , 0 ,, 0 ,,,0.8,-1,,0,
WSPro=,,,, 1 ,,,, 0 ,,,, 0 ,,,,-1 ,-1 ,-1 , 0 , 0 , 0 , 0 , 0
BC Design=,, 0 ,, 0 ,,,,,,

Type RM Length L Ch R = 1 ,27.08   ,8,8,8
BEGIN DESCRIPTION:
È¾´Ü¼öÁ¤
END DESCRIPTION:
#Sta/Elev= 23
       0    4.72    25.7    4.91    35.7    4.82      54    4.97      54       4
   54.85       4   54.85    3.63      56    3.63   61.96     .77   74.86     .77
   76.46    -.03   83.26    -.03   84.86     .77   97.23     .77     102    3.63
  103.15    3.63  103.15       4     104       4     104    4.99   125.8    4.94
   133.8    5.02   142.1    4.91     161     4.7
#Mann= 3 , 0 , 0
       0     .03       0      54     .03       0     104     .03       0
Bank Sta=54,104
Exp/Cntr=0.5,0.3

Type RM Length L Ch R = 1 ,27      ,50,50,50
#Sta/Elev= 27
       0    5.21    34.7    5.03    34.7    4.83    44.2    4.98    50.8    4.83
    50.8    5.03    52.8    5.15    67.5    5.18      71    4.93    74.2    3.64
    80.1     .76   92.97     .76   94.57    -.04  103.37    -.04  104.97     .76
  115.08     .76   121.1    3.57   123.7    4.87     124    4.87   129.2    5.27
   142.6    5.12   144.6    5.02   144.6    4.82   152.6    5.02   160.8    4.87
   160.8    5.07   194.6    5.07
#Mann= 3 , 0 , 0
       0     .03       0      71     .03       0     124     .03       0
Levee=-1,67.5,6,-1,129.2,6,,
Bank Sta=71,124
Exp/Cntr=0.3,0.1

Type RM Length L Ch R = 1 ,26      ,50,50,50
#Sta/Elev= 29
       0    4.89       0    4.79    26.3    4.79    35.8    4.67    35.8    4.87
      50    5.12    56.6    4.94    59.2    3.55   65.34     .71   78.36     .71
   79.96    -.09   86.76    -.09   88.36     .71   99.86     .71   106.2    3.61
   108.3    4.82     109    4.82   116.5    5.37     120    5.37   124.6    5.06
   127.6    5.06   129.6    4.96   129.6    4.76   137.8    4.89   145.7    4.69
   145.7    4.89   147.7    4.89   150.2    5.01   180.2    5.01
#Mann= 3 , 0 , 0
       0     .03       0    56.6     .03       0     109     .03       0
Levee=-1,50,6,-1,116.5,6,,
Bank Sta=56.6,109
Exp/Cntr=0.3,0.1

Type RM Length L Ch R = 1 ,25      ,33,33,33
#Sta/Elev= 30
       0    4.96    33.8    4.96    33.8    4.76    34.3    4.89    40.5    4.89
    49.9    4.66    49.9    4.86    51.9    4.99    65.2    5.03    71.2    4.76
    73.4    3.64   79.71     .66   94.72     .66   96.32    -.14  103.12    -.14
  104.72     .66   114.1     .66   120.2    3.63   122.2    4.95   125.2    5.46
     135    5.46   138.8    4.91     144    4.86     144    4.66   151.8    4.81
   159.9    4.56   159.9    4.76   161.9    4.76   164.1    4.91   195.2    4.91
#Mann= 3 , 0 , 0
       0     .03       0    71.2     .03       0   122.2     .03       0
Levee=-1,65.5,6,-1,125.2,6,,
Bank Sta=71.2,122.2
Exp/Cntr=0.3,0.1

Type RM Length L Ch R = 1 ,24.17   ,17,17,17
#Sta/Elev= 28
       0    4.82       0    4.65     9.4    4.65     9.4    4.85    11.4    4.94
    14.4    4.94    23.7    5.22    30.5    4.87    32.9    3.57    37.8    1.17
    37.8     .62   55.99     .62   57.59    -.18   64.39    -.18   65.99     .62
    75.2     .62    75.2    1.45    79.7    3.57    81.7    4.87    82.7    4.87
    83.7    4.87    89.2    5.37    93.2    5.37    98.2    4.92   101.2    4.87
   103.4    4.62   103.9    4.62   110.7    4.77
#Mann= 3 , 0 , 0
       0     .03       0    30.5     .03       0    81.7     .03       0
Levee=-1,23.7,6,-1,89.2,6,,
Bank Sta=30.5,81.7
Exp/Cntr=0.3,0.1

Type RM Length L Ch R = 1 ,24      ,50,50,50
#Sta/Elev= 30
       0    4.95    33.7    4.85    33.7    4.65    40.4    4.84    49.9    4.66
    49.9    4.86    51.9    4.94    64.5    5.24    71.5    4.86    73.3    3.76
   79.75     .61      97     .61    98.6    -.19   105.4    -.19     107     .61
  113.96     .61   120.1    3.63     122    4.87     126    5.04   129.7    5.36
   132.7    5.36   138.7    4.89   141.7    4.89   143.7    4.76   143.7    4.56
   151.9    4.68   159.8     4.5   159.8     4.7   163.7    4.85   193.7    4.85
#Mann= 3 , 0 , 0
       0     .03       0    71.5     .03       0     122     .03       0
Levee=-1,64.5,6,-1,129.7,6,,
Bank Sta=71.5,122
Exp/Cntr=0.3,0.1

Type RM Length L Ch R = 1 ,23      ,50,50,50
#Sta/Elev= 30
       0    4.92      32    4.88      32    4.68    38.7     4.8    48.1    4.57
    48.1    4.77    50.1    4.94    62.9    5.26    69.8    4.78    71.5    3.58
   77.95     .55    94.2     .55    95.8    -.25   102.6    -.25   104.2     .55
  112.14     .55   118.4    3.57   120.3    4.82   126.7    5.42   131.2    5.42
   136.9    4.87   142.1    4.77   142.1    4.57   149.9    4.72   157.7    4.43
   158.2    4.43   158.2    4.63   160.2    4.63   161.9    4.87   191.9    4.87
#Mann= 3 , 0 , 0
       0     .03       0    69.8     .03       0   120.3     .03       0
Levee=-1,62.9,6,-1,126.7,6,,
Bank Sta=69.8,120.3
Exp/Cntr=0.3,0.1

Type RM Length L Ch R = 1 ,22      ,16,16,16
#Sta/Elev= 30
       0    4.77    33.9    4.77    33.9    4.57    40.7    4.67    50.1    4.52
    50.1    4.72    52.1    4.82    66.7    5.03    71.7    4.64    73.4    3.63
   79.89      .5    93.7      .5    95.3     -.3   102.1     -.3   103.7      .5
     114      .5   120.4    3.46   122.7    4.77   128.2    5.12   132.7    5.12
   138.9    4.87   141.7    4.87   143.7    4.77   143.7    4.57   151.9    4.72
     160    4.57     160    4.77     164    4.77     164    4.57     194    4.57
#Mann= 3 , 0 , 0
       0     .03       0    71.7     .03       0   122.7     .03       0
Levee=-1,66.7,6,-1,128.2,6,,
Bank Sta=71.7,122.7
Exp/Cntr=0.3,0.1

Type RM Length L Ch R = 1 ,21.34   ,25,25,25
#Sta/Elev= 23
       0    4.49    34.3    4.52    41.5    4.49    63.5    4.58    63.5    3.68
    64.5    3.68    64.5    3.07      66    3.07    71.5     .46   82.72     .46
   84.32    -.34   91.12    -.34   92.72     .46  106.11     .46     111    3.17
   112.5    3.17   112.5    3.68   113.5    3.68   113.5    4.58   135.7    4.53
   143.5    4.58   151.6    4.56     172     4.4
#Mann= 3 , 0 , 0
       0     .03       0    63.5     .03       0   113.5     .03       0
Bank Sta=63.5,113.5
Exp/Cntr=0.5,0.3

Type RM Length L Ch R = 3 ,21.215  ,,,
BEGIN DESCRIPTION:
È­Á¤12±³
END DESCRIPTION:
Bridge Culvert--1,0,-1,-1, 0
Deck Dist Width WeirC Skew NumUp NumDn MinLoCord MaxHiCord MaxSubmerge Is_Ogee
0.1,24,1.44,0, 2, 2, , , 0.95, 0, 0,0,,
    63.5   113.5
    4.58    4.58
    3.68    3.68
    63.5   113.5
    4.58    4.58
    3.68    3.68
Pier Skew, UpSta & Num, DnSta & Num=  ,80, 2 ,80, 2 , 0 , 0 , 0 ,,
       1       1
       0       5
       1       1
       0       5
Pier Skew, UpSta & Num, DnSta & Num=  ,97, 2 ,97, 2 , 0 , 0 , 0 ,,
       1       1
       0       5
       1       1
       0       5
BR Coef=-1 , 0 , 0 ,, 0 ,,,0.8,-1,,0,
WSPro=,,,, 1 ,,,, 0 ,,,, 0 ,,,,-1 ,-1 ,-1 , 0 , 0 , 0 , 0 , 0
BC Design=,, 0 ,, 0 ,,,,,,

Type RM Length L Ch R = 1 ,21.09   ,9,9,9
#Sta/Elev= 23
       0    4.49    34.3    4.52    41.5    4.49    63.5    4.58    63.5    3.68
    64.5    3.68    64.5    3.07      66    3.07    71.5     .46   82.72     .46
   84.32    -.34   91.12    -.34   92.72     .46  106.11     .46     111    3.17
   112.5    3.17   112.5    3.68   113.5    3.68   113.5    4.58   135.7    4.53
   143.5    4.58   151.6    4.56     172     4.4
#Mann= 3 , 0 , 0
       0     .03       0    63.5     .03       0   113.5     .03       0
Bank Sta=63.5,113.5
Exp/Cntr=0.5,0.3

Type RM Length L Ch R = 1 ,21      ,50,50,50
#Sta/Elev= 14
       0  5.0023     3.8    4.64     6.5    3.05 11.7595     .45 23.0235     .45
 24.6235    -.35 33.4235    -.35 35.0235     .45 46.4046     .45    52.2    3.22
    54.6    4.64      55    4.64    59.5    4.99      60    4.99
#Mann= 3 , 0 , 0
       0     .03       0     3.8     .03       0    54.6     .03       0
Levee=-1,3.8,4.64,-1,54.6,4.64,,
Bank Sta=3.8,54.6
Exp/Cntr=0.3,0.1

Type RM Length L Ch R = 1 ,20      ,50,50,50
#Sta/Elev= 30
       0    5.37      .7    4.67     2.7    4.67     2.7    4.47    18.7    4.48
    18.7    4.68    20.7     4.8    29.9    5.06    40.6    4.69    42.5    3.31
    49.6    -.14    60.8     .16    61.3    -.45    62.8     -.6    67.8    -.45
    68.3     .09    81.7    -.12    88.6    3.19    90.8    4.76    91.3    4.76
      97    5.16     101    5.16   110.8    4.76   112.8    4.61   112.8    4.41
   120.6    4.56   128.8    4.31   128.8    4.51   130.8    4.51   130.8    4.91
#Mann= 3 , 0 , 0
       0     .03       0    40.6     .03       0    91.3     .03       0
Levee=-1,40.6,5,-1,91.3,5,,
Bank Sta=40.6,91.3
Exp/Cntr=0.3,0.1

Type RM Length L Ch R = 1 ,19      ,38,38,38
#Sta/Elev= 30
       0    5.29      .7    4.59     2.7    4.59     2.7    4.39    18.8     4.4
    18.8     4.6    20.8    4.74    33.7       5    40.5     4.5    42.6     3.2
    49.8    -.15    59.3    -.04    59.8    -.45    60.8    -.65    65.3    -.65
    66.3    -.45    66.8     .05    81.5    -.21    88.8    3.15    90.7     4.6
    91.3     4.6    97.1    5.15   101.6    5.15   107.6     4.7   110.6     4.7
   112.6    4.55   112.6    4.35   113.1     4.5   130.7    4.35   174.1     4.5
#Mann= 3 , 0 , 0
       0     .03       0    40.5     .03       0    91.3     .03       0
Bank Sta=40.5,91.3
Exp/Cntr=0.3,0.1

Type RM Length L Ch R = 1 ,18.12   ,12,12,12
#Sta/Elev= 28
       0    4.54     2.2    4.72     6.6    4.72    21.7    5.13    22.3    5.12
    22.3    3.97    23.3    3.97    23.3    3.58    29.3     .02    41.8    -.04
    42.3    -.46    43.3    -.61    47.8    -.61    48.8    -.46    49.3     -.1
    65.3     -.1    70.3    3.35    71.3    3.35    71.3    3.94    72.3    3.94
    72.3    5.09    92.3    4.62    94.3    4.36   101.5    4.36     102    4.55
   110.2    4.38   113.1    4.68   144.3    4.68
#Mann= 3 , 0 , 0
       0     .03       0    21.7     .03       0    72.3     .03       0
Bank Sta=21.7,72.3
Exp/Cntr=0.3,0.1

Type RM Length L Ch R = 1 ,18      ,50,50,50
#Sta/Elev= 30
       0    5.36       0    4.76     8.4    4.57     8.4    4.37    24.5    4.37
    24.5    4.57    26.5     4.7    34.8    4.82    46.1    4.57    48.2    3.22
    55.5    -.23    64.5    -.01      65    -.46      66    -.61    71.5    -.46
      72     .04    87.2    -.23    96.9    4.42      98    4.94   103.5    5.24
   107.5    5.24   113.3    4.69   118.3    4.59   118.3    4.39   126.2    4.54
   134.5    4.34   134.5    4.54     137    4.54     140    6.84     170    6.84
#Mann= 3 , 0 , 0
       0     .03       0    46.1     .03       0    96.9     .03       0
Bank Sta=46.1,96.9
Exp/Cntr=0.3,0.1

Type RM Length L Ch R = 1 ,17      ,50,50,50
#Sta/Elev= 30
       0    5.74      30    5.74      30    4.44      32    4.44      32    4.24
    48.2    4.23    53.2    4.51      70    4.45      72    3.16      79    -.29
      90    -.14    90.5    -.54      92    -.69    97.5    -.54    97.8    -.19
   111.1    -.31   118.1    3.05   120.2    4.51   120.5    4.51   124.1    4.86
   128.1    4.86   129.8    4.66     140    4.61     142    4.46     142    4.26
   157.9    4.26   157.9    4.46   159.9    4.46   159.9    4.81   190.5    4.81
#Mann= 3 , 0 , 0
       0     .03       0      70     .03       0   120.5     .03       0
Levee=-1,70,5,-1,120.5,5,,
Bank Sta=70,120.5
Exp/Cntr=0.3,0.1

Type RM Length L Ch R = 1 ,16      ,22,22,22
#Sta/Elev= 30
       0    5.82       0    4.52       2    4.52       2    4.32    18.2    4.31
    18.2    4.51    20.2    4.59    33.5    4.86    39.8    4.49      42    3.21
      49    -.21    62.2    -.19    62.5    -.57    65.5    -.87    69.3    -.57
    69.8     -.1      81    -.33    88.3    3.04    90.2    4.44    90.5    4.44
    96.8    4.89     104    4.79     107    4.49   112.2    4.39   112.2    4.19
   128.1    4.19   128.1    4.39   130.1    4.39   130.1    4.74   160.5    4.74
#Mann= 3 , 0 , 0
       0     .03       0    39.8     .03       0    90.5     .03       0
Bank Sta=39.8,90.5
Exp/Cntr=0.3,0.1

Type RM Length L Ch R = 1 ,15.28   ,20,20,20
#Sta/Elev= 20
       0    4.07      56     4.5      56    3.15    57.1    3.15      66    -.09
      72    -.18    76.5    -.19      77    -.58      78    -.73      81    -.73
      83    -.58    83.5     -.2    89.5    -.15   104.9     -.1   104.9    3.22
     106    3.22     106    4.57     135    4.27     144    4.22     165    4.17
#Mann= 3 , 0 , 0
       0     .03       0      56     .03       0     106     .03       0
Levee=-1,56,5,-1,106,5,,
Bank Sta=56,106
Exp/Cntr=0.5,0.3

Type RM Length L Ch R = 3 ,15.18   ,,,
BEGIN DESCRIPTION:
È­Á¤14±³
END DESCRIPTION:
Bridge Culvert--1,0,-1,-1, 0
Deck Dist Width WeirC Skew NumUp NumDn MinLoCord MaxHiCord MaxSubmerge Is_Ogee
0.1,19,1.44,0, 2, 2, , , 0.95, 0, 0,0,,
      56     106
     4.5    4.57
    3.22    3.22
      56     106
     4.5    4.57
    3.22    3.22
Pier Skew, UpSta & Num, DnSta & Num=  ,72, 2 ,72, 2 , 0 , 0 , 0 ,,
     1.2     1.2
       0       4
     1.2     1.2
       0       4
Pier Skew, UpSta & Num, DnSta & Num=  ,89.5, 2 ,89.5, 2 , 0 , 0 , 0 ,,
     1.2     1.2
       0       4
     1.2     1.2
       0       4
BR Coef=-1 , 0 , 0 ,, 0 ,,,0.8,-1,,0,
WSPro=,,,, 1 ,,,, 0 ,,,, 0 ,,,,-1 ,-1 ,-1 , 0 , 0 , 0 , 0 , 0
BC Design=,, 0 ,, 0 ,,,,,,

Type RM Length L Ch R = 1 ,15.08   ,8,8,8
#Sta/Elev= 20
       0    4.07      56     4.5      56    3.15    57.1    3.15      66    -.09
      72    -.18    76.5    -.19      77    -.58      78    -.73      81    -.73
      83    -.58    83.5     -.2    89.5    -.15   104.9     -.1   104.9    3.22
     106    3.22     106    4.57     135    4.27     144    4.22     165    4.17
#Mann= 3 , 0 , 0
       0     .03       0      56     .03       0     106     .03       0
Bank Sta=56,106
Exp/Cntr=0.5,0.3

Type RM Length L Ch R = 1 ,15      ,50,50,50
#Sta/Elev= 30
       0    5.99      30    5.99      30    4.39    31.8    4.39    31.8    4.19
    41.1     4.3    47.9    4.11    47.9    4.31    54.4    4.54    69.1    4.66
    71.4     3.1    78.6    -.35    89.4    -.18      90    -.58    92.9    -.73
    95.4    -.73    96.4    -.58    96.7    -.19     111    -.31   117.9    3.02
   120.4    4.52   124.8    5.02   129.8    5.02   136.7    4.42   141.7    4.32
   141.7    4.12   157.8    4.13   157.8    4.33   159.9    4.33   159.9    4.63
#Mann= 3 , 0 , 0
       0     .03       0    69.1     .03       0   120.4     .03       0
Bank Sta=69.1,120.4
Exp/Cntr=0.3,0.1

Type RM Length L Ch R = 1 ,14      ,50,50,50
#Sta/Elev= 30
       0    5.01    12.7    4.19    19.3    4.33    28.8    4.17    28.8    4.37
    30.8    4.48      43    4.75    50.5    4.31    52.5    3.06    59.5    -.31
    76.4     -.2    77.5    -.82      82    -.82      83     -.6    83.5    -.22
    91.8    -.36    98.8       3     101    4.31     108    4.91   111.5    4.91
   117.7    4.36   122.8    4.26   122.8    4.06   129.5    4.21   138.3    3.96
   138.8    3.96   138.8    4.16   140.8    4.16   140.8    4.61     171    4.61
#Mann= 3 , 0 , 0
       0     .03       0    50.5     .03       0     101     .03       0
Bank Sta=50.5,101
Exp/Cntr=0.3,0.1

Type RM Length L Ch R = 1 ,13      ,50,50,50
#Sta/Elev= 30
       0    5.13      30    5.13      30    4.23      32    4.23      32    4.03
      48    4.03      48    4.23      50    4.38    62.7    4.63    69.7    4.23
    71.8    3.02    78.8    -.32    98.8    -.27    99.3    -.65   100.8    -.75
   105.6    -.65   105.8    -.26     111    -.37   118.1    2.97   120.3    4.23
   128.8    4.88   132.8    4.88   136.9    4.33     142    4.18     142    3.98
   148.6    4.13     158    3.93     158    4.13     160    4.13     160    4.53
#Mann= 3 , 0 , 0
       0     .03       0    69.7     .03       0   120.3     .03       0
Bank Sta=69.7,120.3
Exp/Cntr=0.3,0.1

Type RM Length L Ch R = 1 ,12      ,41,41,41
#Sta/Elev= 30
       0    5.06      30    5.06      30    4.16      32    4.16      32    3.96
    38.7    4.11    48.1    3.96    48.1    4.16    50.1    4.33    63.3    4.69
    69.8    4.21    71.8    3.01    78.9    -.39    93.8    -.34    94.3    -.65
    95.3     -.8     101    -.65   101.8    -.33     111    -.43   120.3    4.21
   127.3    5.01   131.3    5.01     137    4.26   142.1    4.16   142.1    3.96
   148.7    4.11   158.1    3.91   158.1    4.11   160.1    4.11   160.1    4.51
#Mann= 3 , 0 , 0
       0     .03       0    69.8     .03       0   120.3     .03       0
Bank Sta=69.8,120.3
Exp/Cntr=0.3,0.1

Type RM Length L Ch R = 1 ,11.09   ,30,30,30
#Sta/Elev= 23
       0    3.85      57    3.93      57    3.02    57.9    3.02    57.9    2.45
    59.7    2.45    66.2    -.45    73.7    -.41    78.5     -.5      79    -.65
    80.5     -.8      84     -.8    85.5    -.65      86     -.6    90.7    -.55
      98    -.53   104.5    2.46   106.1    2.46   106.1    3.02     107    3.02
     107    3.93     130    3.96     160    3.96
#Mann= 3 , 0 , 0
       0     .03       0      57     .03       0     107     .03       0
Bank Sta=57,107
Exp/Cntr=0.5,0.3

Type RM Length L Ch R = 3 ,10.34   ,,,
BEGIN DESCRIPTION:
È­Á¤15±³
END DESCRIPTION:
Bridge Culvert--1,0,-1,-1, 0
Deck Dist Width WeirC Skew NumUp NumDn MinLoCord MaxHiCord MaxSubmerge Is_Ogee
0.1,29,1.44,0, 2, 2, , , 0.95, 0, 0,0,,
      57     107
    3.93    3.93
    3.02    3.02
      57     107
    3.93    3.93
    3.02    3.02
Pier Skew, UpSta & Num, DnSta & Num=  ,73.7, 2 ,73.7, 2 , 0 , 0 , 0 ,,
       1       1
       0       4
       1       1
       0       4
Pier Skew, UpSta & Num, DnSta & Num=  ,90.7, 2 ,90.7, 2 , 0 , 0 , 0 ,,
       1       1
       0       4
       1       1
       0       4
BR Coef=-1 , 0 , 0 ,, 0 ,,,0.8,-1,,0,
WSPro=,,,, 1 ,,,, 0 ,,,, 0 ,,,,-1 ,-1 ,-1 , 0 , 0 , 0 , 0 , 0
BC Design=,, 0 ,, 0 ,,,,,,

Type RM Length L Ch R = 1 ,10.29   ,12,12,12
#Sta/Elev= 23
       0    3.85      57    3.93      57    3.02    57.9    3.02    57.9    2.45
    59.7    2.45    66.2    -.45    73.7    -.41    78.5     -.5      79    -.65
    80.5     -.8      84     -.8    85.5    -.65      86     -.6    90.7    -.55
      98    -.53   104.5    2.46   106.1    2.46   106.1    3.02     107    3.02
     107    3.93     130    3.96     160    3.96
#Mann= 3 , 0 , 0
       0     .03       0      57     .03       0     107     .03       0
Bank Sta=57,107
Exp/Cntr=0.5,0.3

Type RM Length L Ch R = 1 ,10.17   ,17,17,17
BEGIN DESCRIPTION:
10+17³«Â÷°ø»ó·ù
END DESCRIPTION:
#Sta/Elev= 26
       0    7.16      30    7.16      40    4.66    40.7    4.13    42.7    4.13
    42.7    3.93      52    4.04    58.7    3.97    58.7    4.17    60.8    4.31
    63.8    4.31      72    4.56    80.5    4.08    83.5    2.42    89.7    -.65
     122    -.65   127.9    2.45     131    3.76   137.3    4.33   150.5    4.21
   152.5    4.08   152.5    3.88     162    4.02   168.7     3.9   168.7     4.1
   175.7     4.2
#Mann= 3 , 0 , 0
       0     .03       0    80.5     .03       0     131     .03       0
Bank Sta=80.5,131
Exp/Cntr=0.3,0.1

Type RM Length L Ch R = 1 ,10      ,50,50,50
#Sta/Elev= 30
       0     5.8      30     5.8      30     3.8      32     3.8      32     3.6
    41.5     3.8    48.2    3.75    48.2    3.95    50.2     4.1      61     4.4
    69.9     3.7    79.4     -.8    83.7     -.8    84.2   -1.15    86.2   -1.55
    99.2    -1.6   106.2   -1.15   106.7    -.78   110.7    -.78   117.3    2.33
   119.7     3.6   121.7     3.6   129.7    4.45   142.2    4.15   142.2    3.95
   151.5    4.05   158.2    3.95   158.2    4.15   165.7    4.55   195.7    4.55
#Mann= 3 , 0 , 0
       0     .03       0    69.9     .03       0   119.7     .03       0
Bank Sta=69.9,119.7
Exp/Cntr=0.3,0.1

Type RM Length L Ch R = 1 ,9       ,50,50,50
#Sta/Elev= 30
       0    5.99      30    5.99      30    3.99      32    3.99      32    3.79
    41.5    3.99    48.1    3.89    48.1    4.09    50.1    4.24    63.1    4.39
    69.4    3.97    72.9    2.44    79.1    -.71    83.1    -.71    84.6    -1.3
   105.8    -1.3   106.3   -1.15   106.8    -.79   110.8    -.79   119.8    3.59
   120.4    3.79   127.2    4.59   131.7    4.59     137    4.19   141.9    4.09
   141.9    3.89   150.1    3.99   158.2    3.94   176.1    4.49   206.1    4.49
#Mann= 3 , 0 , 0
       0     .03       0    69.4     .03       0   120.4     .03       0
Bank Sta=69.4,120.4
Exp/Cntr=0.3,0.1

Type RM Length L Ch R = 1 ,8       ,33,33,33
#Sta/Elev= 30
       0    6.33      30    6.33      30    4.33      32    4.33      32    4.13
    38.7    4.29    48.1    4.09    48.1    4.29    53.1    4.39    56.6    4.69
    64.4    4.59    69.4    4.09    79.1    -.66    83.1    -.66    83.9   -1.16
    85.6   -1.36   100.6   -1.41   106.1   -1.16   106.6    -.76   110.6    -.76
   120.1    3.89   128.6    4.69   141.9    4.14   141.9    3.94   148.7    4.09
   158.3    3.84   158.3    4.04   160.3    4.04   160.3    4.94   190.3    4.94
#Mann= 3 , 0 , 0
       0     .03       0    69.4     .03       0   120.1     .03       0
Bank Sta=69.4,120.1
Exp/Cntr=0.3,0.1

Type RM Length L Ch R = 1 ,7.17    ,17,17,17
#Sta/Elev= 30
       0    5.73      30    5.73      31    4.03      33    4.03      33    3.83
    49.2    3.87    49.2    4.07    51.2    4.23      66    4.43    70.5    4.04
    76.7    1.04    76.7    -.56    84.6    -.73    84.6   -1.16    85.5   -1.31
     106   -1.31     107   -1.16   107.2    -.71   115.1    -.65   115.1     .95
   121.5    3.83   130.3    4.68   133.3    4.68     143    4.03     143    3.83
   159.1    3.78   159.1    3.98   161.1    3.98   161.1    4.98   191.1    4.98
#Mann= 3 , 0 , 0
       0     .03       0    70.5     .03       0   121.5     .03       0
Bank Sta=70.5,121.5
Exp/Cntr=0.3,0.1

Type RM Length L Ch R = 1 ,7       ,50,50,50
#Sta/Elev= 30
       0    4.21    15.2    3.83    21.5       4      31    3.82      31    4.02
      33    4.19    45.7    4.46    52.5    4.08    55.8    2.18    62.1    -.72
    66.1    -.72    66.8   -1.16    67.3   -1.36    88.5   -1.46      89   -1.16
      90    -.77      94    -.77     100    2.16     103    3.86   112.8    4.77
   115.8    4.77     120    4.11     125    4.01     125    3.81   131.6    3.96
     141    3.79     141    3.99     143    3.99     143    4.99     173    4.99
#Mann= 3 , 0 , 0
       0     .03       0    52.5     .03       0     103     .03       0
Bank Sta=52.5,103
Exp/Cntr=0.3,0.1

Type RM Length L Ch R = 1 ,6       ,50,50,50
#Sta/Elev= 30
       0    5.46      30    5.46      30    3.96      32    3.96      32    3.76
    38.6    3.96    48.2     3.8    48.2       4    50.2    4.15    63.1    4.38
    69.8    3.86    79.2    -.86    83.2    -.86    84.2   -1.56   101.7   -1.51
   105.4   -1.36   106.4     -.8   110.9     -.8   117.1    2.09   120.2    3.91
   129.7    4.71   132.7    4.71     137    4.11   141.9    4.01   141.9    3.81
     158    3.81     158    4.01   160.1    4.01   160.1    4.91   190.1    4.91
#Mann= 3 , 0 , 0
       0     .03       0    69.8     .03       0   120.2     .03       0
Bank Sta=69.8,120.2
Exp/Cntr=0.3,0.1

Type RM Length L Ch R = 1 ,5       ,50,50,50
#Sta/Elev= 30
       0    5.44      30    5.44      30    3.94    31.7    3.94    31.7    3.74
    38.2    3.94    47.7    3.78    47.7    3.98    49.7    4.09      63    4.44
    69.2     3.8    72.4    2.14    82.5    -.72    83.7   -1.56   105.2   -1.46
   106.6    -.71   110.6    -.79   116.6    2.09   119.7    3.74   127.3    4.49
   132.7    4.54   136.5    4.09   141.5    3.99   141.5    3.79   148.3    3.94
   157.7    3.79   157.7    4.01   159.7    4.01   159.7    5.01   189.7    5.01
#Mann= 3 , 0 , 0
       0     .03       0    69.2     .03       0   119.7     .03       0
Bank Sta=69.2,119.7
Exp/Cntr=0.3,0.1

Type RM Length L Ch R = 1 ,4       ,10,10,10
#Sta/Elev= 28
       0    5.57      30    5.57      30    3.87    31.7    3.87    31.7    3.67
    38.4    3.77    47.8    3.67    47.8    3.87    49.8    3.96    68.4    4.08
    78.7    -.76    82.7    -.76    83.8   -1.52   105.3   -1.57   106.3    -.83
   110.7    -.83     117    1.97   119.7    3.38   126.7    4.06   139.8    3.94
   141.8    3.86   141.8    3.66   148.3    3.83   157.7    3.63   157.7    3.83
   159.7    3.83   159.7    4.83   189.7    4.83
#Mann= 3 , 0 , 0
       0     .03       0    68.4     .03       0   119.7     .03       0
Bank Sta=68.4,119.7
Exp/Cntr=0.3,0.1

Type RM Length L Ch R = 1 ,3.40    ,20,20,20
#Sta/Elev= 30
       0    3.71    47.3    3.66    47.3    2.79    48.2    2.79    48.2    1.59
    49.2    1.59    49.2     .59    53.1     .59    57.5    -.79      61    -.79
    61.5   -1.17      64   -1.57    71.6   -1.57    83.5   -1.13      84    -.72
    88.5    -.72    91.7     .67    95.6     .63    95.6    1.64    96.6    1.64
    96.6    2.84    97.5    2.84    97.5    3.71   120.2    3.76   127.3    3.88
   135.5    3.69   135.5    3.89   137.5    3.89   137.5    4.99   167.5    4.99
#Mann= 3 , 0 , 0
       0     .03       0    47.3     .03       0    97.5     .03       0
Bank Sta=47.3,97.5
Exp/Cntr=0.5,0.3

Type RM Length L Ch R = 3 ,3.30    ,,,
BEGIN DESCRIPTION:
È­Á¤16±³
END DESCRIPTION:
Bridge Culvert--1,0,-1,-1, 0
Deck Dist Width WeirC Skew NumUp NumDn MinLoCord MaxHiCord MaxSubmerge Is_Ogee
0.1,19,1.44,0, 2, 2, , , 0.95, 0, 0,0,,
    47.3    97.5
    3.66    3.71
    2.79    2.84
    47.3    97.5
    3.66    3.71
    2.79    2.84
Pier Skew, UpSta & Num, DnSta & Num=  ,64, 2 ,64, 2 , 0 , 0 , 0 ,,
       1       1
       0     4.5
       1       1
       0     4.5
Pier Skew, UpSta & Num, DnSta & Num=  ,81, 2 ,81, 2 , 0 , 0 , 0 ,,
       1       1
       0     4.5
       1       1
       0     4.5
BR Coef=-1 , 0 , 0 ,, 0 ,,,0.8,-1,,0,
WSPro=,,,, 1 ,,,, 0 ,,,, 0 ,,,,-1 ,-1 ,-1 , 0 , 0 , 0 , 0 , 0
BC Design=,, 0 ,, 0 ,,,,,,

Type RM Length L Ch R = 1 ,3.20    ,20,20,20
#Sta/Elev= 30
       0    3.71    47.3    3.66    47.3    2.79    48.2    2.79    48.2    1.59
    49.2    1.59    49.2     .59    53.1     .59    57.5    -.79      61    -.79
    61.5   -1.17      64   -1.57    71.6   -1.57    83.5   -1.13      84    -.72
    88.5    -.72    91.7     .67    95.6     .63    95.6    1.64    96.6    1.64
    96.6    2.84    97.5    2.84    97.5    3.71   120.2    3.76   127.3    3.88
   135.5    3.69   135.5    3.89   137.5    3.89   137.5    4.99   167.5    4.99
#Mann= 3 , 0 , 0
       0     .03       0    47.3     .03       0    97.5     .03       0
Bank Sta=47.3,97.5
Exp/Cntr=0.5,0.3

Type RM Length L Ch R = 1 ,3       ,50,50,50
#Sta/Elev= 29
       0    5.23    17.4    5.16    17.4    5.36      29    5.12    31.7    5.04
    36.5    3.94    53.5    3.83    57.6    1.76    63.3    -.79    67.3    -.79
    67.8   -1.17    69.3   -1.67    89.2   -1.47    90.2    -.82    94.7    -.82
   100.2    1.76   103.2     3.4     104    3.71   111.6    4.11   116.6    4.22
   120.9    3.92     126    3.84     126    3.64   132.5    3.81   141.9    3.63
   141.9    3.83     144    3.83     144    4.86     174    4.86
#Mann= 3 , 0 , 0
       0     .03       0    53.5     .03       0     104     .03       0
Bank Sta=53.5,104
Exp/Cntr=0.3,0.1

Type RM Length L Ch R = 1 ,2       ,50,50,50
#Sta/Elev= 30
       0    6.15      30    6.15    34.9    5.56    34.9    6.41    35.3    6.41
    35.3    5.41    42.4    5.32      46    4.21    62.9    3.99    73.2    -.73
    77.7    -.73      78   -1.17    79.5   -1.77    98.4   -1.67    98.9   -1.17
    99.4    -.83   103.9    -.83   109.8    2.02   113.2    3.85   120.9    4.54
     125    4.62   130.2    4.07   135.3    3.95   135.3    3.75   141.8    3.92
   151.3    3.76   151.3    3.96   153.5    3.96   153.5    4.96   183.5    4.96
#Mann= 3 , 0 , 0
       0     .03       0    62.9     .03       0   113.2     .03       0
Bank Sta=62.9,113.2
Exp/Cntr=0.3,0.1

Type RM Length L Ch R = 1 ,1       ,50,50,50
#Sta/Elev= 29
       0    4.46     5.2    4.46    18.2    6.01    30.7    5.66    36.6    4.41
    42.2    4.41    43.3    4.84    53.2    3.93    62.7    -.65    67.2    -.65
    67.7   -1.18    73.2   -1.78    87.2   -1.78    89.2   -1.18    89.9    -.69
      94    -.69   102.7    3.49   103.2    3.81   111.7    4.56   116.2    4.56
   120.2    4.11   125.4    4.01   125.4    3.79   132.5    3.96   141.2    3.76
   141.2    3.97   143.4    3.97   143.4    4.97   173.4    4.97
#Mann= 3 , 0 , 0
       0     .03       0    53.2     .03       0   103.2     .03       0
Bank Sta=53.2,103.2
Exp/Cntr=0.3,0.1

Type RM Length L Ch R = 1 ,0       ,0,0,0
#Sta/Elev= 25
       0    4.07    27.1    3.83    30.5    2.02    36.4    -.79    44.4    -.64
    44.9   -1.18    47.4   -1.98    54.4   -1.98    64.1   -1.98    66.1   -1.18
    66.6    -.77    70.9    -.84    76.5    1.93    79.4    3.37    80.1    3.74
    86.5    4.47    93.1    4.53    97.5    4.04   100.6    3.97   102.5     3.9
   102.5     3.7     103     3.7   111.6    3.88   129.8    3.74   159.8    3.74
#Mann= 3 , 0 , 0
       0     .03       0    27.1     .03       0    79.4     .03       0
Bank Sta=27.1,79.4
Exp/Cntr=0.3,0.1

Chan Stop Cuts=-1
Use User Specified Reach Order=0
User Specified Reach Order=RIVER-1         ,Reach-1
