HEC-RAS study Hwajung.prj: Hwajung

--- Hwajung.g01 (geometry) --- (continued)

Type RM Length L Ch R = 1 ,72      ,50,50,50
#Sta/Elev= 27
       0    8.68    33.6    8.68    33.6    7.57    36.5    7.44    36.5    7.29
      43    7.48    52.1    7.27    53.6    7.47    59.8     4.7    69.2    4.33
    71.3    3.84      76    3.66    76.5    3.66    76.6    3.76    77.8    4.31
    87.2    4.63    91.4    6.58    93.6    7.39    96.6    7.39    96.6    7.19
    97.1    7.19   103.4    7.44   109.7    7.39   113.3    7.49   113.3    7.64
   115.8    7.73   145.8    7.73
#Mann= 3 , 0 , 0
       0     .03       0    53.6     .03       0    93.6     .03       0
Levee=-1,53.6,9,-1,93.6,9,,
Bank Sta=53.6,93.6
Exp/Cntr=0.3,0.1

Type RM Length L Ch R = 1 ,71      ,43,43,43
#Sta/Elev= 30
       0    8.98      30    8.98      30    7.68    32.8    7.57    32.8    7.37
    39.6    7.63    46.9    7.45    46.9    7.65    49.9     7.8    49.9    7.43
    56.2    4.61    66.1    4.23    66.9    3.69    68.7    3.59    70.7    3.59
    72.5    3.69    73.7    4.19    83.7    4.51    87.7    6.41    88.6    7.05
    89.3    7.05    89.3     7.5    92.6     7.5    92.6     7.3    99.7    7.55
   106.5    7.42   106.5    7.62   109.4    7.69   110.7    8.89   140.7    8.89
#Mann= 3 , 0 , 0
       0     .03       0    49.9     .03       0    89.3     .03       0
Levee=-1,49.9,9,-1,89.3,9,,
Bank Sta=49.9,89.3
Exp/Cntr=0.3,0.1

Type RM Length L Ch R = 1 ,70.07   ,35,35,35
#Sta/Elev= 23
       0    8.22      15    8.07    36.5    8.07    36.5    7.27    37.5    7.27
    37.5    5.81    40.5    4.61    47.5    4.21    50.5    4.01    51.5    3.66
      52    3.56      55    3.56    57.5    3.56      58    3.66      59    4.06
    61.5    4.36    68.5    4.51      71    5.95      71    7.27      72    7.27
      72    8.07      75    8.07   116.5    7.83
#Mann= 3 , 0 , 0
       0     .03       0    36.5     .03       0      72     .03       0
Levee=-1,36.5,9,-1,72,9,,
Bank Sta=36.5,72
Exp/Cntr=0.5,0.3

Type RM Length L Ch R = 3 ,69.395  ,,,
BEGIN DESCRIPTION:
È­Á¤3±³
END DESCRIPTION:
Bridge Culvert--1,0,-1,-1, 0
Deck Dist Width WeirC Skew NumUp NumDn MinLoCord MaxHiCord MaxSubmerge Is_Ogee
0.1,34,1.44,0, 2, 2, , , 0.95, 0, 0,0,,
    36.5      72
    8.07    8.07
    7.27    7.27
    36.5      72
    8.07    8.07
    7.27    7.27
Pier Skew, UpSta & Num, DnSta & Num=  ,47.5, 2 ,47.5, 2 , 0 , 0 , 0 ,,
      .6      .6
     3.5       8
      .6      .6
     3.5       8
Pier Skew, UpSta & Num, DnSta & Num=  ,61.5, 2 ,61.5, 2 , 0 , 0 , 0 ,,
      .6      .6
     3.5       8
      .6      .6
     3.5       8
BR Coef=-1 , 0 , 0 ,, 0 ,,,0.8,-1,,0,
WSPro=,,,, 1 ,,,, 0 ,,,, 0 ,,,,-1 ,-1 ,-1 , 0 , 0 , 0 , 0 , 0
BC Design=,, 0 ,, 0 ,,,,,,

Type RM Length L Ch R = 1 ,69.22   ,22,22,22
#Sta/Elev= 23
       0    8.22      15    8.07    36.5    8.07    36.5    7.27    37.5    7.27
    37.5    5.81    40.5    4.61    47.5    4.21    50.5    4.01    51.5    3.66
      52    3.56      55    3.56    57.5    3.56      58    3.66      59    4.06
    61.5    4.36    68.5    4.51      71    5.95      71    7.27      72    7.27
      72    8.07      75    8.07   116.5    7.83
#Mann= 3 , 0 , 0
       0     .03       0    36.5     .03       0      72     .03       0
Levee=-1,36.5,9,-1,72,9,,
Bank Sta=36.5,72
Exp/Cntr=0.5,0.3

Type RM Length L Ch R = 1 ,69      ,50,50,50
#Sta/Elev= 29
       0    7.83      30    7.83    32.9    7.73    32.9    7.53    39.2    7.64
    46.9    7.57    46.9    7.77    49.9    7.77    49.9    7.42    55.6    4.99
    62.7    4.37    63.9    3.89    70.7    3.65    71.2     3.5    71.7     3.5
    73.5    3.94      85    3.75      85     4.1    86.7     4.1    86.7     6.5
    89.8    7.84    92.8    7.84    92.8    7.64    93.3    7.64    99.7    7.76
   106.7    7.69   106.7    7.89   109.7    7.95   139.7    7.95
#Mann= 3 , 0 , 0
       0     .03       0    49.9     .03       0    89.8     .03       0
Levee=-1,49.9,9,-1,89.8,9,,
Bank Sta=49.9,89.8
Exp/Cntr=0.3,0.1

Type RM Length L Ch R = 1 ,68      ,47,47,47
#Sta/Elev= 28
       0    7.24      30    7.24    33.1    7.21    33.1    7.01    39.9     7.2
    46.6    6.97    48.5    7.04    48.5    7.24      50    7.24    52.3    6.34
      56     4.4    66.4    3.92    67.2     3.5    68.6     3.4    70.8     3.4
    72.9     3.5      74    3.98    83.9    4.51    86.9    5.81      89    7.35
      93    7.35      93    7.15     100    7.28     107    7.12     107    7.32
   110.1    7.38   112.6    8.68   142.6    8.68
#Mann= 3 , 0 , 0
       0     .03       0      50     .03       0      89     .03       0
Levee=-1,50,9,-1,89,9,,
Bank Sta=50,89
Exp/Cntr=0.3,0.1

Type RM Length L Ch R = 1 ,67.03   ,4,4,4
#Sta/Elev= 28
       0    7.72      30    7.72    32.5    7.42    35.5     7.4    35.5     7.2
    42.5    7.33    49.7    7.12    51.2    7.47    51.2    7.32    52.7    7.32
    53.8     6.5    58.4    4.23    67.4    4.44    68.4    3.47    69.8    3.36
    75.3    3.36      76    3.47      77    4.44    86.1    4.46    92.1    7.22
    92.8    7.47    95.8    7.47    95.8    7.27   102.4     7.4   109.6    7.25
   109.6    7.45   112.3     7.5     113     8.2
#Mann= 3 , 0 , 0
       0     .03       0    52.7     .03       0    92.8     .03       0
Levee=-1,52.7,9,-1,92.8,9,,
Bank Sta=52.7,92.8
Exp/Cntr=0.3,0.1

Type RM Length L Ch R = 1 ,66.49   ,49,49,49
#Sta/Elev= 28
       0    7.72      30    7.72    32.5    7.42    35.5     7.4    35.5     7.2
    42.5    7.33    49.7    7.12    51.2    7.47    51.2    7.32    52.7    7.32
    53.8     6.5    58.4    4.23    67.4    4.44    68.4    3.47    69.8    3.36
    75.3    3.36      76    3.47      77    4.44    86.1    4.46    92.1    7.22
    92.8    7.47    95.8    7.47    95.8    7.27   102.4     7.4   109.6    7.25
   109.6    7.45   112.3     7.5     113     8.2
#Mann= 3 , 0 , 0
       0     .03       0    52.7     .03       0    92.8     .03       0
Levee=-1,52.7,9,-1,92.8,9,,
Bank Sta=52.7,92.8
Exp/Cntr=0.3,0.1

Type RM Length L Ch R = 1 ,66      ,50,50,50
#Sta/Elev= 30
       0    7.36      30    7.36    32.5    7.16    35.5    7.09    35.5    6.84
    42.3    7.05    49.4     6.9    50.9    6.96    50.9    7.16    52.4    7.16
    53.1    7.16    54.3    6.48    58.8     4.2    68.6    3.86    69.2    3.43
    70.8    3.28    72.8    3.28    75.3    3.43    76.1    3.88    85.9    4.19
    92.3    7.19    92.8    7.19    95.3    7.19    95.3    6.99   102.4    7.19
   109.3    6.99   109.3    7.19   112.1    7.24   113.1    8.04   143.1    8.04
#Mann= 3 , 0 , 0
       0     .03       0    52.4     .03       0    92.8     .03       0
Levee=-1,52.4,9,-1,92.8,9,,
Bank Sta=52.4,92.8
Exp/Cntr=0.3,0.1

Type RM Length L Ch R = 1 ,65      ,37,37,37
#Sta/Elev= 28
       0    7.52      30    7.52      36    7.13      36    6.98      43    7.21
    50.3    7.03    50.3    7.23    53.1    7.26    55.1    6.19    59.1    4.52
    68.5    4.09    69.5     3.4    72.4    3.25    75.5    3.25    76.2     3.4
      77    3.89    86.5    4.04    92.6    7.14    92.9    7.49    93.6    7.49
    95.9    7.49    95.9    7.39    96.4    7.39     103    7.53   109.9     7.4
     113    7.59     114    8.09     144    8.09
#Mann= 3 , 0 , 0
       0     .03       0    53.1     .03       0    93.6     .03       0
Levee=-1,53.1,9,-1,93.6,9,,
Bank Sta=53.1,93.6
Exp/Cntr=0.3,0.1

Type RM Length L Ch R = 1 ,64.13   ,20,20,20
#Sta/Elev= 23
       0    8.34    77.8    7.84    77.8    7.04    78.8    7.04    78.8    6.22
    83.3    4.09    90.3    3.77    93.3    3.66    93.8    3.38    94.8    3.18
    97.8    3.18   101.8    3.18   102.3    3.38   103.8    3.62   106.8    3.81
   113.3    4.65   116.8    5.66   116.8    7.03   117.8    7.03   117.8    7.83
   131.8    7.83   141.3    7.29   160.9     7.2
#Mann= 3 , 0 , 0
       0     .03       0    77.8     .03       0   117.8     .03       0
Levee=-1,77.8,9,-1,117.8,9,,
Bank Sta=77.8,117.8
Exp/Cntr=0.5,0.3

Type RM Length L Ch R = 3 ,64.03   ,,,
BEGIN DESCRIPTION:
È­Á¤2±³
END DESCRIPTION:
Bridge Culvert--1,0,-1,-1, 0
Deck Dist Width WeirC Skew NumUp NumDn MinLoCord MaxHiCord MaxSubmerge Is_Ogee
0.1,19,1.44,0, 2, 2, , , 0.95, 0, 0,0,,
    77.8   117.8
    7.84    7.84
    7.04    7.04
    77.8   117.8
    7.84    7.84
    7.04    7.04
Pier Skew, UpSta & Num, DnSta & Num=  ,90.3, 2 ,90.3, 2 , 0 , 0 , 0 ,,
      .6      .6
       3     8.7
      .6      .6
       3     8.7
Pier Skew, UpSta & Num, DnSta & Num=  ,105.3, 2 ,105.3, 2 , 0 , 0 , 0 ,,
      .6      .6
       3     8.7
      .6      .6
       3     8.7
BR Coef=-1 , 0 , 0 ,, 0 ,,,0.8,-1,,0,
WSPro=,,,, 1 ,,,, 0 ,,,, 0 ,,,,-1 ,-1 ,-1 , 0 , 0 , 0 , 0 , 0
BC Design=,, 0 ,, 0 ,,,,,,

Type RM Length L Ch R = 1 ,63.43   ,43,43,43
#Sta/Elev= 23
       0    8.34    77.8    7.84    77.8    7.04    78.8    7.04    78.8    6.22
    83.3    4.09    90.3    3.77    93.3    3.66    93.8    3.38    94.8    3.18
    97.8    3.18   101.8    3.18   102.3    3.38   103.8    3.62   106.8    3.81
   113.3    4.65   116.8    5.66   116.8    7.03   117.8    7.03   117.8    7.83
   131.8    7.83   141.3    7.29   160.9     7.2
#Mann= 3 , 0 , 0
       0     .03       0    77.8     .03       0   117.8     .03       0
Levee=-1,77.8,9,-1,117.8,9,,
Bank Sta=77.8,117.8
Exp/Cntr=0.5,0.3

Type RM Length L Ch R = 1 ,63      ,15,15,15
#Sta/Elev= 27
       0    9.83      30    9.83      30    7.43    32.8    7.15    39.8    7.35
    47.3    7.06    50.4    7.42    50.4    6.77    52.1    6.29    56.7     3.9
    65.8    4.09    66.8    3.36    70.9    3.26    78.3    3.36    79.4    4.07
    83.9    4.13    87.8    6.11    89.7     6.9    89.7    7.35    92.6    7.35
    92.6    7.15    99.7     7.2     106    7.05   106.5    7.05   106.5    7.25
   109.9     7.3   139.9     7.3
#Mann= 3 , 0 , 0
       0     .03       0    50.4     .03       0    89.7     .03       0
Levee=-1,50.4,8,-1,89.7,8,,
Bank Sta=50.4,89.7
Exp/Cntr=0.3,0.1

Type RM Length L Ch R = 1 ,62.35   ,35,35,35
#Sta/Elev= 30
       0    9.25      30    9.25      30    7.25    32.9    7.22    32.9    7.02
    39.7    7.26    46.6       7    47.1       7    47.1     7.2    50.1     7.2
    56.5       4    63.1     3.9    64.7     3.2    65.2     3.1    65.7     3.2
    66.6    4.01    73.6    3.91    75.2     3.2    76.7       3    78.8     3.2
    80.5    3.95      84    4.26    88.2    6.16    89.7    7.18    92.7    7.18
    92.7    6.88    99.6    7.08   106.9    6.99   106.9    7.18   140.2    7.18
#Mann= 3 , 0 , 0
       0     .03       0    50.1     .03       0    89.7     .03       0
Levee=-1,50.1,8,-1,89.7,8,,
Bank Sta=50.1,89.7
Exp/Cntr=0.3,0.1

Type RM Length L Ch R = 1 ,62      ,50,50,50
#Sta/Elev= 28
       0    9.12      30    9.12      38    8.32    39.5    8.32    39.5    7.11
    42.6    7.06    42.6    6.86    49.5    7.12    56.5    6.93    56.5    7.13
    59.5    7.19    65.8    4.01      79    3.85    80.5    3.53    85.5    2.96
    87.7    2.96    89.2    3.96    93.3    4.08      97    5.91    99.2    7.12
   102.2    7.12   102.2    6.92   109.3    7.02   116.4    6.87   116.4    7.07
   119.5    7.12   121.2    7.37   151.2    7.37
#Mann= 3 , 0 , 0
       0     .03       0    59.5     .03       0    99.2     .03       0
Levee=-1,59.5,8,-1,99.2,8,,
Bank Sta=59.5,99.2
Exp/Cntr=0.3,0.1

Type RM Length L Ch R = 1 ,61      ,37,37,37
#Sta/Elev= 27
       0    8.19      30    8.19      30    6.96    32.8    6.97    32.8    6.77
    39.7    7.05    46.9    6.74    46.9    6.94      50    7.05      52    5.92
    55.9    4.18    70.9    3.73    72.5    3.02    73.6    2.92    77.5    3.02
    78.5    3.65    83.6    3.99    89.9    7.09    92.9    7.09    92.9    6.89
    99.7    7.04   106.6    6.88   106.6    7.08   109.8    7.08   111.4    7.33
   111.7    7.59   141.7    7.59
#Mann= 3 , 0 , 0
       0     .03       0      50     .03       0    89.9     .03       0
Levee=-1,50,8,-1,89.9,8,,
Bank Sta=50,89.9
Exp/Cntr=0.3,0.1

Type RM Length L Ch R = 1 ,60.13   ,4,4,4
#Sta/Elev= 27
       0    7.38      30    7.38    31.5    7.13    34.6    6.98    34.6    6.78
    41.5    6.97    48.6    6.97    48.6    7.17    51.6    7.17    57.4    3.91
    70.7     3.8    71.7    3.02    72.7    2.87    79.2    2.87    79.7    3.02
    80.7     3.8    85.4    3.87    89.4    6.11    91.4    7.09    94.4    7.09
    94.4    6.89   101.4    7.02   108.4     6.8   108.4       7   112.8    7.09
   113.4    7.36   143.4    7.36
#Mann= 3 , 0 , 0
       0     .03       0    51.6     .03       0    91.4     .03       0
Levee=-1,51.6,8,-1,91.4,8,,
Bank Sta=51.6,91.4
Exp/Cntr=0.3,0.1

Type RM Length L Ch R = 1 ,60.09   ,9,9,9
#Sta/Elev= 27
       0    7.38      30    7.38    31.5    7.13    34.6    6.98    34.6    6.78
    41.5    6.97    48.6    6.97    48.6    7.17    51.6    7.17    57.4    3.91
    70.7     3.8    71.7    3.02    72.7    2.87    79.2    2.87    79.7    3.02
    80.7     3.8    85.4    3.87    89.4    6.11    91.4    7.09    94.4    7.09
    94.4    6.89   101.4    7.02   108.4     6.8   108.4       7   112.8    7.09
   113.4    7.36   143.4    7.36
#Mann= 3 , 0 , 0
       0     .03       0    51.6     .03       0    91.4     .03       0
Levee=-1,51.6,8,-1,91.4,8,,
Bank Sta=51.6,91.4
Exp/Cntr=0.3,0.1

Type RM Length L Ch R = 1 ,60      ,50,50,50
#Sta/Elev= 28
       0    7.25      30    7.25      32       7    34.9    6.95    34.9    6.75
    41.9    6.95      49     6.7      49     6.9    52.1    7.05    53.7    6.15
    58.5       4    72.7     3.9    73.2    3.55    74.2    3.02    75.2    2.92
    77.6    2.92    79.7    3.02    81.4     3.7    85.5    3.85    91.9    7.05
    94.9    7.05    94.9    6.85     102       7   108.9     6.8   108.9       7
   111.9       7   113.5    7.15   123.7    7.65
#Mann= 3 , 0 , 0
       0     .03       0    52.1     .03       0    91.9     .03       0
Levee=-1,52.1,8,-1,91.9,8,,
Bank Sta=52.1,91.9
Exp/Cntr=0.3,0.1

Type RM Length L Ch R = 1 ,59      ,50,50,50
#Sta/Elev= 28
       0    7.09      30    7.09      33    6.84      36    6.72      36    6.57
      43    6.83    50.1    6.61    50.1    6.81      53    6.91    54.9    5.93
    59.4    3.95    73.6    3.71    74.1    3.56    74.9       3    78.5    2.85
    80.4       3    81.9    3.52    86.9    3.84    91.3    5.98    92.8    6.86
    95.8    6.76    95.8    6.56   102.9    6.71   109.9    6.66   109.9    6.86
     115    6.91   119.5    6.51   149.5    6.51
#Mann= 3 , 0 , 0
       0     .03       0      53     .03       0    92.8     .03       0
Levee=-1,53,8,-1,92.8,8,,
Bank Sta=53,92.8
Exp/Cntr=0.3,0.1

Type RM Length L Ch R = 1 ,58      ,50,50,50
#Sta/Elev= 26
       0    6.78      30    6.78      32    6.68    35.2    6.36    35.2    6.54
    42.2     6.7    49.2    6.47    49.2    6.67    52.2    6.78    54.1    5.71
    57.9    3.98    72.7     3.7    73.2    3.55    74.1       3    76.2     2.8
    78.6     2.8    80.3       3    81.3    3.59    86.1    3.81    89.6    5.34
    91.9     6.8    94.9     6.8    94.9    6.55   108.9    6.59   108.9    6.79
   141.9    6.79
#Mann= 3 , 0 , 0
       0     .03       0    52.2     .03       0    91.9     .03       0
Levee=-1,52.2,8,-1,91.9,8,,
Bank Sta=52.2,91.9
Exp/Cntr=0.3,0.1

Type RM Length L Ch R = 1 ,57      ,32,32,32
#Sta/Elev= 29
       0    6.82      30    6.82      32    6.57    34.9     6.6    34.9     6.4
    41.8     6.6    48.9    6.39    48.9    6.59    51.9    6.68    57.3    4.08
    72.4    3.68      73    3.58    73.9    2.98    76.3    2.68    77.9    2.68
    80.1    2.98    80.8    3.61    85.7    3.77    89.3     5.4    91.6    6.72
    94.6    6.72    94.6    6.52   101.5    6.61   108.5    6.54   108.5    6.74
   111.4    6.84   114.8    6.77   125.4    3.81   155.4    3.81
#Mann= 3 , 0 , 0
       0     .03       0    51.9     .03       0    91.6     .03       0
Levee=-1,51.9,8,-1,91.6,8,,
Bank Sta=51.9,91.6
Exp/Cntr=0.3,0.1

Type RM Length L Ch R = 1 ,56.18   ,3.3,3.3,3.3
#Sta/Elev= 27
       0    6.84      30    6.84    35.5    6.59    35.5    6.39    42.5    6.67
    49.4     6.4    49.4    6.65    52.5    6.78    54.3    5.69    58.3    3.88
      72    3.79    73.1    2.98    73.6    2.77    80.1    2.77    81.1    2.98
      82    3.79    86.3     3.8    90.3    6.01    92.3    6.77    95.3    6.52
   102.2    6.61   109.2    6.54   109.2    6.74   112.1    6.84   115.5    6.77
   126.1    3.81   156.1    3.81
#Mann= 3 , 0 , 0
       0     .03       0    52.5     .03       0    92.3     .03       0
Levee=-1,52.5,8,-1,92.3,8,,
Bank Sta=52.5,92.3
Exp/Cntr=0.3,0.1

Type RM Length L Ch R = 1 ,56.147  ,14.7,14.7,14.7
#Sta/Elev= 27
       0    6.84      30    6.84    35.5    6.59    35.5    6.39    42.5    6.67
    49.4     6.4    49.4    6.65    52.5    6.78    54.3    5.69    58.3    3.88
      72    3.79    73.1    2.98    73.6    2.77    80.1    2.77    81.1    2.98
      82    3.79    86.3     3.8    90.3    6.01    92.3    6.77    95.3    6.52
   102.2    6.61   109.2    6.54   109.2    6.74   112.1    6.84   115.5    6.77
   126.1    3.81   156.1    3.81
#Mann= 3 , 0 , 0
       0     .03       0    52.5     .03       0    92.3     .03       0
Levee=-1,52.5,8,-1,92.3,8,,
Bank Sta=52.5,92.3
Exp/Cntr=0.3,0.1

Type RM Length L Ch R = 1 ,56      ,50,50,50
#Sta/Elev= 30
       0    6.67    32.5    6.67    35.3    6.53    35.3    6.39    35.8    6.39
    42.4    6.63    49.3     6.4    49.3     6.6    52.3     6.7      54     5.8
    58.4    3.85    72.6    3.58    73.6    3.47    74.5    2.98    75.8    2.88
    80.5    2.98    81.3    3.57    86.4     3.8    90.3    5.69    92.1    6.68
    95.1    6.63    95.1    6.43    95.6    6.43   102.1    6.58     109    6.52
     109    6.73   114.1    6.72   122.6    4.64   124.6    3.84   127.6    3.54
#Mann= 3 , 0 , 0
       0     .03       0    52.3     .03       0    92.1     .03       0
Levee=-1,52.3,8,-1,92.1,8,,
Bank Sta=52.3,92.1
Exp/Cntr=0.3,0.1

Type RM Length L Ch R = 1 ,55      ,50,50,50
#Sta/Elev= 30
       0    6.69      30    6.69    35.5    6.51    35.5    6.36    42.6    6.49
      49     6.3    49.5     6.3    49.5     6.5    52.5    6.56    54.3    5.53
    57.9    3.94    72.7     3.6    73.9     3.5    74.6    2.98    76.5    2.68
    78.2    2.68    80.6    2.98    81.2    3.48    86.4    3.69    92.2    6.65
    92.7    6.65    95.2     6.6    95.2     6.4    95.7     6.4   102.2    6.61
   109.2    6.48   109.2    6.67   114.4    6.71   125.7    4.05   155.7    4.05
#Mann= 3 , 0 , 0
       0     .03       0    52.5     .03       0    92.7     .03       0
Levee=-1,52.5,8,-1,92.7,8,,
Bank Sta=52.5,92.7
Exp/Cntr=0.3,0.1

Type RM Length L Ch R = 1 ,54      ,50,50,50
#Sta/Elev= 30
       0    6.84      32    6.84      32    6.54      35    6.54      35    6.34
      42     6.6    48.6    6.28    49.1    6.28    49.1    6.48      52    6.64
    53.5    5.72    57.1    4.07    72.3    3.58    73.4    3.48    74.1    2.97
    75.3    2.72    77.8    2.72    80.2    2.97    80.9    3.48    86.3    3.83
    91.8    6.61    92.3    6.61    94.8    6.51    94.8    6.31    95.3    6.31
   101.8    6.56   108.9    6.44   108.9    6.64   117.5    6.72     122    4.66
#Mann= 3 , 0 , 0
       0     .03       0      52     .03       0    92.3     .03       0
Levee=-1,52,8,-1,92.3,8,,
Bank Sta=52,92.3
Exp/Cntr=0.3,0.1

Type RM Length L Ch R = 1 ,53      ,2.1,2.1,2.1
#Sta/Elev= 28
       0     6.6      30     6.6    33.1    6.23    33.6    6.23    40.4    6.48
    47.4    6.59    47.4    6.79    50.3    6.79    50.3    6.95    50.5    6.95
    50.5    6.34    52.1    3.75    70.9    3.73      72    2.97    73.6    2.82
    76.3    2.82      79    2.97    80.1     3.7    89.9     3.9    89.9    6.85
    90.4    6.85    92.9    6.85    92.9    6.65    99.8    6.72   106.8    6.59
   106.8    6.79   110.2    6.85   121.5    6.68
#Mann= 3 , 0 , 0
       0     .03       0    50.3     .03       0    90.4     .03       0
Levee=-1,50.3,8,-1,90.4,8,,
Bank Sta=50.3,90.4
Exp/Cntr=0.3,0.1

Type RM Length L Ch R = 1 ,52.479  ,20.9,20.9,20.9
#Sta/Elev= 30
       0    6.48      30    6.48      30    6.28    30.5    6.28    52.5    6.83
    52.5    5.33    53.5    5.33    53.5    3.85      65     3.7      73    3.71
    73.5    3.71    74.5    2.97      75    2.73    77.5    2.69      82    2.83
    82.5    2.97      83    3.26    91.5    3.45    91.5    5.28    92.5    5.28
    92.5    6.78      93    6.78   102.4    6.33   108.6    6.28   109.1    6.28
   109.1    6.48   112.8    6.54   116.2    6.58   117.2    6.58   122.7    4.54
#Mann= 3 , 0 , 0
       0     .03       0    52.5     .03       0      93     .03       0
Levee=-1,52.5,8,-1,93,8,,
Bank Sta=52.5,93
Exp/Cntr=0.5,0.3

Type RM Length L Ch R = 3 ,52.3745 ,,,
BEGIN DESCRIPTION:
È­¶û±³
END DESCRIPTION:
Bridge Culvert--1,0,-1,-1, 0
Deck Dist Width WeirC Skew NumUp NumDn MinLoCord MaxHiCord MaxSubmerge Is_Ogee
0.1,20,1.44,0, 2, 2, , , 0.95, 0, 0,0,,
    52.5    92.5
    6.83    6.78
    5.33    5.28
    52.5    92.5
    6.83    6.78
    5.33    5.28
Pier Skew, UpSta & Num, DnSta & Num=  ,65, 2 ,65, 2 , 0 , 0 , 0 ,,
      .7      .7
       2       7
      .7      .7
       2       7
Pier Skew, UpSta & Num, DnSta & Num=  ,80, 2 ,80, 2 , 0 , 0 , 0 ,,
      .7      .7
       2       7
      .7      .7
       2       7
BR Coef=-1 , 0 , 0 ,, 0 ,,,0.8,-1,,0,
WSPro=,,,, 1 ,,,, 0 ,,,, 0 ,,,,-1 ,-1 ,-1 , 0 , 0 , 0 , 0 , 0
BC Design=,, 0 ,, 0 ,,,,,,

Type RM Length L Ch R = 1 ,52.27   ,10,10,10
#Sta/Elev= 30
       0    6.48      30    6.48      30    6.28    30.5    6.28    52.5    6.83
    52.5    5.33    53.5    5.33    53.5    3.85      65     3.7      73    3.71
    73.5    3.71    74.5    2.97      75    2.73    77.5    2.69      82    2.83
    82.5    2.97      83    3.26    91.5    3.45    91.5    5.28    92.5    5.28
    92.5    6.78      93    6.78   102.4    6.33   108.6    6.28   109.1    6.28
   109.1    6.48   112.8    6.54   116.2    6.58   117.2    6.58   122.7    4.54
#Mann= 3 , 0 , 0
       0     .03       0    52.5     .03       0      93     .03       0
Levee=-1,52.5,8,-1,93,8,,
Bank Sta=52.5,93
Exp/Cntr=0.5,0.3

Type RM Length L Ch R = 1 ,52.17   ,3.3,3.3,3.3
#Sta/Elev= 23
       0    7.35      30    7.35      30    6.35    32.8    6.14    39.9    6.34
    46.9    6.19    49.9     6.5    56.7     3.9    70.2    3.45    71.2    2.95
    73.2    2.85    76.2    2.85    78.2    2.97    79.2    3.45    83.7    3.56
    87.7    5.56    89.7    6.42    90.2    6.42   106.4    6.17     110     6.4
   115.6    6.45   122.5    4.54   124.2    3.54
#Mann= 3 , 0 , 0
       0     .03       0    49.9     .03       0    90.2     .03       0
Levee=-1,49.9,8,-1,90.2,8,,
Bank Sta=49.9,90.2
Exp/Cntr=0.3,0.1

Type RM Length L Ch R = 1 ,52.137  ,13.7,13.7,13.7
#Sta/Elev= 23
       0    7.35      30    7.35      30    6.35    32.8    6.14    39.9    6.34
    46.9    6.19    49.9     6.5    56.7     3.9    70.2    3.45    71.2    2.95
    73.2    2.85    76.2    2.85    78.2    2.97    79.2    3.45    83.7    3.56
    87.7    5.56    89.7    6.42    90.2    6.42   106.4    6.17     110     6.4
   115.6    6.45   122.5    4.54   124.2    3.54
#Mann= 3 , 0 , 0
       0     .03       0    49.9     .03       0    90.2     .03       0
Levee=-1,49.9,8,-1,90.2,8,,
Bank Sta=49.9,90.2
Exp/Cntr=0.3,0.1

Type RM Length L Ch R = 1 ,52      ,31,31,31
#Sta/Elev= 26
       0    7.52    31.5    7.52    31.5    6.62    34.5    6.42    34.5    6.22
    41.5    6.43    48.5    6.25    48.5    6.45    51.5    6.47    56.3    4.07
    71.5    3.62    72.4    2.97      74    2.82    78.1    2.82    80.2    2.97
      81    3.56    85.5    3.67    91.3    6.47    91.5    6.47    94.3    6.47
    94.3    6.27   101.2    6.44   108.2    6.25   108.2    6.45   117.5    6.52
   123.5    4.63
#Mann= 3 , 0 , 0
       0     .03       0    51.5     .03       0    91.5     .03       0
Levee=-1,51.5,8,-1,91.5,8,,
Bank Sta=51.5,91.5
Exp/Cntr=0.3,0.1

Type RM Length L Ch R = 1 ,51.19   ,19,19,19
#Sta/Elev= 30
       0     6.6      30     6.6    32.9    6.42    32.9    6.22      40    6.43
    46.3    6.13    46.8    6.13    46.8    6.33    49.9    6.44    55.1    4.07
    63.9    3.75    65.7    2.84      66    2.94    66.3    3.47    74.3    3.56
      76    2.94    79.8    2.94    80.2    3.57    83.7    3.63    89.7    6.47
    90.2    6.47    92.7    6.37    93.2    6.17   106.6    6.21   106.6    6.41
   111.7    6.51   113.8    6.27   121.7    4.63   123.2    3.73   153.2    3.73
#Mann= 3 , 0 , 0
       0     .03       0    49.9     .03       0    90.2     .03       0
Levee=-1,49.9,8,-1,90.2,8,,
Bank Sta=49.9,90.2
Exp/Cntr=0.3,0.1

Type RM Length L Ch R = 1 ,51      ,50,50,50
#Sta/Elev= 30
       0    6.78      30    6.78    35.1    6.38    35.1    6.18      42    6.37
      49    6.12      49    6.32      52     6.4    57.4       4    71.1    3.54
      72    2.82    74.5    2.67    78.8    2.67    81.2    2.82    81.8    3.35
    86.1    3.54    91.8    6.45      92    6.45    94.8    6.35    94.8    6.15
    95.3    6.15   101.8    6.28   108.7    6.19   108.7    6.39   111.3    6.54
   113.8    6.49   115.9    6.25   123.8    4.61   125.3    3.71   155.3    3.71
#Mann= 3 , 0 , 0
       0     .03       0      52     .03       0      92     .03       0
Levee=-1,52,8,-1,92,8,,
Bank Sta=52,92
Exp/Cntr=0.3,0.1

Type RM Length L Ch R = 1 ,50      ,37,37,37
#Sta/Elev= 29
       0    7.27    31.4    7.27    31.4    6.26    34.5    6.23    34.5    6.03
    41.7    6.28    48.6    6.03    48.6    6.23    51.5    6.39    57.2    3.64
    73.9    3.36    74.7    2.79    79.3    2.64    80.7    2.79      82    3.37
    85.5    3.51    91.3    6.37    91.5    6.37    94.3    6.27    94.3    6.07
    94.8    6.07   101.4     6.3   108.2    6.18   108.2    6.37   113.2    6.42
   123.6    4.65   125.5    3.85   126.5    3.65   156.5    3.65
#Mann= 3 , 0 , 0
       0     .03       0    51.5     .03       0    91.5     .03       0
Levee=-1,51.5,8,-1,91.5,8,,
Bank Sta=51.5,91.5
Exp/Cntr=0.3,0.1

Type RM Length L Ch R = 1 ,49.13   ,3.5,3.5,3.5
#Sta/Elev= 30
       0    7.43    31.7    7.43    31.7    6.43    34.6    6.37    34.6    6.17
    41.6    6.71    48.1    6.12    48.6    6.12    48.6    6.32    51.6    6.41
    57.6    3.52    73.6    3.47    74.6    2.79    76.6    2.59    81.6    2.79
    82.6    3.47    86.1    3.49    90.1    5.34    91.6    6.35    92.1    6.35
    94.6    6.35    94.6    6.15    95.1    6.15   108.2    6.19   108.2    6.39
   111.1    6.52   113.4    6.41   124.2    4.63   126.4    3.83   156.4    3.83
#Mann= 3 , 0 , 0
       0     .03       0    51.6     .03       0    92.1     .03       0
Levee=-1,51.6,8,-1,92.1,8,,
Bank Sta=51.6,92.1
Exp/Cntr=0.3,0.1

Type RM Length L Ch R = 1 ,49.095  ,9.5,9.5,9.5
#Sta/Elev= 30
       0    7.43    31.7    7.43    31.7    6.43    34.6    6.37    34.6    6.17
    41.6    6.71    48.1    6.12    48.6    6.12    48.6    6.32    51.6    6.41
    57.6    3.52    73.6    3.47    74.6    2.79    76.6    2.59    81.6    2.79
    82.6    3.47    86.1    3.49    90.1    5.34    91.6    6.35    92.1    6.35
    94.6    6.35    94.6    6.15    95.1    6.15   108.2    6.19   108.2    6.39
   111.1    6.52   113.4    6.41   124.2    4.63   126.4    3.83   156.4    3.83
#Mann= 3 , 0 , 0
       0     .03       0    51.6     .03       0    92.1     .03       0
Levee=-1,51.6,8,-1,92.1,8,,
Bank Sta=51.6,92.1
Exp/Cntr=0.3,0.1

Type RM Length L Ch R = 1 ,49      ,50,50,50
#Sta/Elev= 28
       0    7.43    32.7    7.43    32.7    6.43    35.7    6.26    35.7    6.06
    42.8    6.38    49.7    6.17    49.7    6.37    52.7    6.45    58.2     3.7
    75.3    3.37    75.8    2.79    77.4    2.59    80.2    2.59      82    2.79
    82.6    3.28    86.7    3.62    92.5    6.35    95.4    6.33    95.4    6.13
   102.4    6.32   109.3    6.13   109.3    6.33   112.3    6.48   114.5    6.39
   123.5    4.66   125.5    4.06   155.5    4.06
#Mann= 3 , 0 , 0
       0     .03       0    52.7     .03       0    92.5     .03       0
Levee=-1,52.7,8,-1,92.5,8,,
Bank Sta=52.7,92.5
Exp/Cntr=0.3,0.1

Type RM Length L Ch R = 1 ,48      ,50,50,50
#Sta/Elev= 29
       0    6.71    31.7    6.71    31.7    6.41    34.6    6.24    34.6    6.04
    41.8    6.34    48.3    6.13    48.8    6.13    48.8    6.33    51.8    6.34
    57.3    3.71    73.7    3.28    74.5    2.78    76.3    2.63    78.7    2.63
    80.6    2.78    81.4    3.33    85.8    3.57    88.8    4.87    91.6    6.36
    91.8    6.36    94.6    6.36    94.6    6.16   101.6     6.2   108.1    5.96
   108.6    5.96   108.6    6.16   111.1     6.2   163.1    6.23
#Mann= 3 , 0 , 0
       0     .03       0    51.8     .03       0    91.8     .03       0
Levee=-1,51.8,7,-1,91.8,7,,
Bank Sta=51.8,91.8
Exp/Cntr=0.3,0.1

Type RM Length L Ch R = 1 ,47      ,50,50,50
#Sta/Elev= 30
       0    7.26      30    7.26      30    6.26    32.5    6.11    32.5    5.91
    39.2    6.23    46.5    5.97    46.5    6.17    49.5    6.28    54.8    3.71
      69    3.51    70.6    3.41    72.1    2.75    73.7     2.6      78    2.75
    78.7     3.3      84    3.71    87.8    5.49      89    6.18    89.7    6.26
    92.2    6.26    92.2    6.06   105.6    5.99   106.1    5.99   106.1    6.19
     111    6.18   111.5    5.74   112.2    5.74   112.9    6.41   142.9    6.41
#Mann= 3 , 0 , 0
       0     .03       0    49.5     .03       0    89.7     .03       0
Levee=-1,49.5,7,-1,89.7,7,,
Bank Sta=49.5,89.7
Exp/Cntr=0.3,0.1

Type RM Length L Ch R = 1 ,46      ,50,50,50
#Sta/Elev= 30
       0    8.06      30    8.06      31    7.96      31     6.1    34.1    6.01
    34.1    5.76    41.2    6.02      48    5.84      48    6.04    50.9    6.12
    56.1    3.61    70.8     3.3    71.5    3.25      73    2.71    74.5    2.56
    78.9    2.71    79.9    3.27    85.1    3.43      91    6.16    93.8    6.06
    93.8    5.86    94.3    5.86   100.9    6.01   107.7    5.91   107.7    6.11
   112.7    6.21   113.5    5.61   114.5    5.61     115    6.31     145    6.31
#Mann= 3 , 0 , 0
       0     .03       0    50.9     .03       0      91     .03       0
Levee=-1,50.9,7,-1,91,7,,
Bank Sta=50.9,91
Exp/Cntr=0.3,0.1

Type RM Length L Ch R = 1 ,45      ,50,50,50
#Sta/Elev= 29
       0    6.43      30    6.43    31.9    6.11    34.8    5.85    41.8    6.09
      49    5.87      52    6.12    53.8    5.07    56.7    3.63    73.8    3.27
    74.8     2.7    75.8     2.6    78.4     2.7    79.9    2.92    81.2    3.26
    86.1    3.46    90.1    5.19    91.6    5.96    94.6    5.96    94.6    5.76
   101.6    5.86   108.5    5.81   108.5    6.01   111.5    6.01   113.3    6.26
   114.1    5.66   115.1    5.66   116.1    6.31   146.1    6.31
#Mann= 3 , 0 , 0
       0     .03       0      52     .03       0    91.6     .03       0
Levee=-1,52,7,-1,91.6,7,,
Bank Sta=52,91.6
Exp/Cntr=0.3,0.1

Type RM Length L Ch R = 1 ,44      ,50,50,50
#Sta/Elev= 30
       0     7.9      30     7.9      30     6.3      33    5.96    39.9    6.23
      47    5.99      47    6.19    50.1    6.23    50.1    5.83    51.7    5.12
    58.8     3.6    71.6    3.25      73    2.63    74.9    2.53    78.5    2.75
    79.5    3.18    84.5    3.43    88.6    5.29    90.1     5.7    90.1       6
    90.2       6    93.6     5.7    99.7       6   106.9     5.9   106.9     6.1
   111.7     6.4   112.1     5.9   113.1     5.9   113.7    6.25   143.7    6.25
#Mann= 3 , 0 , 0
       0     .03       0    50.1     .03       0    90.2     .03       0
Levee=-1,50.1,7,-1,90.2,7,,
Bank Sta=50.1,90.2
Exp/Cntr=0.3,0.1

Type RM Length L Ch R = 1 ,43      ,50,50,50
#Sta/Elev= 30
       0    8.25      30    8.25      30    6.55      33    6.32      33    6.12
    39.9    6.39    46.3    6.16    46.9    6.16    46.9    6.41    49.9    6.37
    49.9    5.97    54.8    3.48    70.2    3.22      71    3.15    73.4     2.5
    78.1     2.6    79.1    3.17      84    3.33    89.7    5.97    89.7    6.42
    90.2    6.42    92.7    6.32    92.7    6.12    99.9    6.22   106.7    6.11
   106.7    6.31   109.8    6.41   111.6    6.72   111.8    6.58   141.8    6.58
#Mann= 3 , 0 , 0
       0     .03       0    49.9     .03       0    90.2     .03       0
Levee=-1,49.9,6.37,-1,90.2,6.42,,
Bank Sta=49.9,90.2
Exp/Cntr=0.3,0.1

Type RM Length L Ch R = 1 ,42      ,4.7,4.7,4.7
#Sta/Elev= 22
       0    7.73    41.6    6.88    71.7    6.73    71.7    6.17    72.5    6.17
    72.5    4.67      75    3.69      85    3.51      89    2.54    89.5    2.44
      93    2.44      94    2.45    94.5    2.54      96     3.4      98    3.43
     106    3.41   109.2    4.47   109.2    6.12     110    6.12     110    6.77
     113    6.72   156.1    6.55
#Mann= 3 , 0 , 0
       0     .03       0    71.7     .03       0     110     .03       0
Bank Sta=71.7,110
Exp/Cntr=0.3,0.1

Type RM Length L Ch R = 1 ,41.453  ,43.3,43.3,43.3
#Sta/Elev= 22
       0    7.73    41.6    6.88    71.7    6.73    71.7    6.17    72.5    6.17
    72.5    4.67      75    3.69      85    3.51      89    2.54    89.5    2.44
      93    2.44      94    2.45    94.5    2.54      96     3.4      98    3.43
     106    3.41   109.2    4.47   109.2    6.12     110    6.12     110    6.77
     113    6.72   156.1    6.55
#Mann= 3 , 0 , 0
       0     .03       0    71.7     .03       0     110     .03       0
Bank Sta=71.7,110
Exp/Cntr=0.5,0.3

Type RM Length L Ch R = 3 ,41.2365 ,,,
BEGIN DESCRIPTION:
È­Á¤1±³
END DESCRIPTION:
Bridge Culvert--1,0,-1,-1, 0
Deck Dist Width WeirC Skew NumUp NumDn MinLoCord MaxHiCord MaxSubmerge Is_Ogee
0.1,43,1.44,0, 2, 2, , , 0.95, 0, 0,0,,
    71.7     110
    6.73    6.73
    6.17    6.17
    71.7     110
    6.73    6.73
    6.17    6.17
Pier Skew, UpSta & Num, DnSta & Num=  ,85, 2 ,85, 2 , 0 , 0 , 0 ,,
       1       1
       2       7
       1       1
       2       7
Pier Skew, UpSta & Num, DnSta & Num=  ,98, 2 ,98, 2 , 0 , 0 , 0 ,,
       1       1
       2       7
       1       1
       2       7
BR Coef=-1 , 0 , 0 ,, 0 ,,,0.8,-1,,0,
WSPro=,,,, 1 ,,,, 0 ,,,, 0 ,,,,-1 ,-1 ,-1 , 0 , 0 , 0 , 0 , 0
BC Design=,, 0 ,, 0 ,,,,,,

Type RM Length L Ch R = 1 ,41.02   ,2,2,2
#Sta/Elev= 22
       0    7.73    41.6    6.88    71.7    6.73    71.7    6.17    72.5    6.17
    72.5    4.67      75    3.69      85    3.51      89    2.54    89.5    2.44
      93    2.44      94    2.45    94.5    2.54      96     3.4      98    3.43
     106    3.41   109.2    4.47   109.2    6.12     110    6.12     110    6.77
     113    6.72   156.1    6.55
#Mann= 3 , 0 , 0
       0     .03       0    71.7     .03       0     110     .03       0
Bank Sta=71.7,110
Exp/Cntr=0.5,0.3

Type RM Length L Ch R = 1 ,41      ,50,50,50
#Sta/Elev= 25
       0    7.48     5.2     6.9      13    6.62    24.5    6.66    31.5    6.48
    35.2    6.81    35.2    5.81    36.5    4.91    39.8    3.24    47.8    3.17
    49.8    2.49    54.3    2.39    60.7    2.49    62.2    2.99    69.2    2.93
    74.3    5.55    74.5    5.55    74.5    6.15    77.5    6.05    77.5    5.85
      88    6.06    98.5    5.87    98.5    6.07   103.5    6.15     109    7.42
#Mann= 3 , 0 , 0
       0     .03       0    35.2     .03       0    74.5     .03       0
Levee=-1,35.2,6.81,-1,74.5,6.15,,
Bank Sta=35.2,74.5
Exp/Cntr=0.3,0.1

Type RM Length L Ch R = 1 ,40      ,50,50,50
#Sta/Elev= 28
       0    7.88     9.7    7.24    13.4    6.21    16.6    6.14    16.6    5.94
    17.1    5.94    27.1    6.13    33.6    5.91    34.1    5.91    34.1    6.06
      37    6.13    42.4    3.28    46.3    3.21    47.8    2.48    56.3    2.33
    61.3    2.33    66.9    2.48    69.2    3.46    71.2    3.46    74.4    4.85
    76.3    5.93    76.8    5.98    79.8    5.88    79.8    5.68    80.3    5.68
    87.5    5.88   101.1    5.88   133.3    6.83
#Mann= 3 , 0 , 0
       0     .03       0      37     .03       0    76.8     .03       0
Levee=-1,37,6.13,-1,76.8,5.98,,
Bank Sta=37,76.8
Exp/Cntr=0.3,0.1

Type RM Length L Ch R = 1 ,39      ,50,50,50
#Sta/Elev= 30
       0    7.87       7    7.23    15.3    5.86    18.4    5.84    18.4    5.64
    25.6    5.78    32.4    5.57    32.4    5.77    35.6    5.86    40.4    3.18
    44.7    3.19    48.4    2.34    48.7    2.44    49.1    2.98    52.6    2.87
    53.4    2.54    62.2    2.44    62.8    2.24    66.3    2.44    66.6    2.75
    69.4    3.25    74.5    5.67    75.3    5.77    78.1    5.67    78.1    5.47
    88.5    5.69    99.2     5.5    99.2     5.7   104.2    5.73   110.7    6.97
#Mann= 3 , 0 , 0
       0     .03       0    35.6     .03       0    75.3     .03       0
Levee=-1,35.6,7,-1,75.3,7,,
Bank Sta=35.6,75.3
Exp/Cntr=0.3,0.1

Type RM Length L Ch R = 1 ,38      ,21,21,21
#Sta/Elev= 26
       0    6.53       0    5.89    13.5    5.87    13.5    5.67    23.6    5.86
    30.5    5.61    30.5    5.81    33.7    5.91    35.7    5.08    39.1    3.26
      49    3.03    50.7    2.39    52.7    2.19    58.6    2.19    62.7    2.39
    63.3    2.79    68.2    3.72    71.2    4.72    72.7    5.81    76.7    5.71
    76.7    5.51    86.7    5.66    97.5    5.43    97.5    5.63   102.4    5.66
     112    7.52
#Mann= 3 , 0 , 0
       0     .03       0    33.7     .03       0    72.7     .03       0
Levee=-1,33.7,5.91,-1,72.7,5.81,,
Bank Sta=33.7,72.7
Exp/Cntr=0.3,0.1

Type RM Length L Ch R = 1 ,37.29   ,4,4,4
#Sta/Elev= 30
       0    6.38    40.5    5.71    50.6     5.8    57.1    5.52    57.6    5.52
    57.6    5.72    60.6    5.73    63.2    5.07    66.7    3.08    76.7    2.99
    76.7    2.35    76.7    2.25    81.2    2.25    84.7    2.25    84.7    2.35
    84.7    2.99    94.7    3.18    98.2    4.73   100.2     5.6   101.2     5.6
   103.2    5.55   103.2    5.35   103.7    5.35   113.4     5.5   123.7    5.34
   124.2    5.34   124.2    5.54   127.1    5.59   129.1    5.59   140.2    7.31
#Mann= 3 , 0 , 0
       0     .03       0    60.6     .03       0   100.2     .03       0
Levee=-1,60.6,7,-1,100.2,7,,
Bank Sta=60.6,100.2
Exp/Cntr=0.3,0.1

Type RM Length L Ch R = 1 ,37.25   ,25,25,25
#Sta/Elev= 30
       0    6.38    40.5    5.71    50.6     5.8    57.1    5.52    57.6    5.52
    57.6    5.72    60.6    5.73    63.2    5.07    66.7    3.08    76.7    2.99
    76.7    2.35    76.7    2.25    81.2    2.25    84.7    2.25    84.7    2.35
    84.7    2.99    94.7    3.18    98.2    4.73   100.2     5.6   101.2     5.6
   103.2    5.55   103.2    5.35   103.7    5.35   113.4     5.5   123.7    5.34
   124.2    5.34   124.2    5.54   127.1    5.59   129.1    5.59   140.2    7.31
#Mann= 3 , 0 , 0
       0     .03       0    60.6     .03       0   100.2     .03       0
Levee=-1,60.6,7,-1,100.2,7,,
Bank Sta=60.6,100.2
Exp/Cntr=0.3,0.1

Type RM Length L Ch R = 1 ,37      ,50,50,50
#Sta/Elev= 25
       0    6.19       0    5.81    15.9    5.61    23.2    5.73    30.2    5.56
    30.2    5.76    33.2    5.91      38    3.36    51.1    3.17    51.8    2.58
    52.7    2.34      54    2.19    57.5    2.14    59.3    2.34    60.3     2.6
    60.8    3.15    66.9    3.03    72.6    5.71    75.6    5.61    75.6    5.41
    86.1     5.6    96.7    5.41    96.7    5.61   101.5    5.71   111.7    6.88
#Mann= 3 , 0 , 0
       0     .03       0    33.2     .03       0    72.6     .03       0
Levee=-1,33.2,5.91,-1,72.6,5.71,,
Bank Sta=33.2,72.6
Exp/Cntr=0.3,0.1

Type RM Length L Ch R = 1 ,36      ,50,50,50
#Sta/Elev= 30
       0    8.96       0    6.46      13    6.27    24.1     5.7    27.1    5.66
    27.1    5.46    37.2    5.65      44    5.38      44    5.58    47.2    5.71
    47.9    5.55    48.9    4.89    51.8    3.36      63    3.28    63.4    2.29
    64.2    2.19    71.7    2.19    73.2    2.43    73.6    2.98      81    2.85
    86.6    5.65    87.2    5.65    89.6    5.55    89.6    5.35    99.7    5.51
   110.8    5.21   110.8    5.41     114     5.5   125.1    6.25   147.2    6.73
#Mann= 3 , 0 , 0
       0     .03       0    47.2     .03       0    87.2     .03       0
Levee=-1,47.2,5.71,-1,87.2,5.65,,
Bank Sta=47.2,87.2
Exp/Cntr=0.3,0.1

Type RM Length L Ch R = 1 ,35      ,50,50,50
#Sta/Elev= 29
       0    6.71      33    6.18    33.8     5.5    36.5    5.49      37    5.29
      47    5.49    53.9    5.36    53.9    5.56    57.1    5.59    58.8    4.69
    62.8       3      75    2.75    78.4    2.25    80.3     2.1    83.3     2.1
    85.1    2.25    87.1    2.94      91    3.01    96.3    5.66    96.8    5.66
    99.3    5.56    99.3    5.36   106.8    5.61   117.3    5.28   117.3    5.48
   123.3    5.55   139.8    6.26   139.8    6.06   157.6    6.49
#Mann= 3 , 0 , 0
       0     .03       0    57.1     .03       0    96.8     .03       0
Levee=-1,57.1,5.59,-1,96.8,5.66,,
Bank Sta=57.1,96.8
Exp/Cntr=0.3,0.1

Type RM Length L Ch R = 1 ,34      ,20,20,20
#Sta/Elev= 30
       0    8.47    35.4    6.86    36.4    5.75    39.6    5.53    39.6    5.33
    49.6    5.62    56.5    5.43    56.5    5.58    59.7    5.71      65    3.08
    70.1    2.77      71    1.97    71.6    2.61    73.9    1.97    74.6    2.12
    75.1    2.74    85.4    2.72    85.9    2.12      88    2.12    89.9    3.01
      94    3.04    99.4    5.62   102.4    5.57   102.4    5.37   109.6    5.62
   123.2    5.32   123.2    5.52   128.3    5.62   132.9    7.37   162.9    7.37
#Mann= 3 , 0 , 0
       0     .03       0    59.7     .03       0    99.4     .03       0
Levee=-1,59.7,5.71,-1,99.4,5.62,,
Bank Sta=59.7,99.4
Exp/Cntr=0.3,0.1

Type RM Length L Ch R = 1 ,33.3    ,30,30,30
#Sta/Elev= 30
       0    8.69    34.5    7.04    35.8    5.71    38.9    5.64    38.9    5.44
      49     5.6    56.1    5.38    56.1    5.58    59.1    5.63    60.6    5.01
    64.3    3.09    73.4    2.64      74    1.97    74.3    2.12    74.5    2.56
    75.4    2.56    75.7    2.12    76.5    1.97    84.5    1.97    87.3    3.07
    93.3    3.26    98.5    5.74   101.5    5.64   101.5    5.44   108.7    5.74
   122.3    5.44   122.3    5.64   127.4    5.74     132    7.49     162    7.49
#Mann= 3 , 0 , 0
       0     .03       0    59.1     .03       0    98.5     .03       0
Bank Sta=59.1,98.5
Exp/Cntr=0.3,0.1

Type RM Length L Ch R = 1 ,33      ,42,42,42
#Sta/Elev= 30
       0    8.57    34.3    7.05    35.4     5.9    38.5    5.83    38.5    5.63
    48.7    5.73    55.6    5.53    55.6    5.73    58.7    5.85      64    2.88
    73.5    2.28    73.8    1.82    74.2    1.82    74.5    2.25      75    2.25
    75.5    1.82    76.5    1.62    79.5    1.62    80.7    1.82    81.6    2.23
      84    2.82    93.1    3.12      98    5.76     101    5.69     101    5.49
   108.2    5.74   118.6    5.54   118.6    5.74     127    5.94   160.1    7.48
#Mann= 3 , 0 , 0
       0     .03       0    58.7     .03       0      98     .03       0
Bank Sta=58.7,98
Exp/Cntr=0.3,0.1

Type RM Length L Ch R = 1 ,32.08   ,70,70,70
#Sta/Elev= 24
       0    6.87    36.2    6.58    43.3    6.79    50.8    6.67      55    6.75
      55    6.15    55.6    6.15    55.6    4.77      61    1.35    68.5    1.45
      71    1.02    74.5    1.04    75.5    1.48    86.5    1.46    89.4     3.8
    89.4    6.05      90    6.05      90    6.65   103.2    6.45   112.9    6.17
   113.4    6.17   113.4    6.37   117.8     6.5   149.5     6.5
#Mann= 3 , 0 , 0
       0     .03       0      55     .03       0      90     .03       0
Bank Sta=55,90
Exp/Cntr=0.3,0.1

Type RM Length L Ch R = 3 ,31.23   ,,,
BEGIN DESCRIPTION:
È­Á¤±³
END DESCRIPTION:
Bridge Culvert--1,0,-1,-1, 0
Deck Dist Width WeirC Skew NumUp NumDn MinLoCord MaxHiCord MaxSubmerge Is_Ogee
0.1,69,1.44,0, 2, 2, , , 0.95, 0, 0,0,,
      55      90
    6.75    6.65
    6.15    6.05
    39.5    74.5
    6.58    6.58
    5.98    5.98
Pier Skew, UpSta & Num, DnSta & Num=  ,65.5, 2 ,50, 2 , 0 , 0 , 0 ,,
      .6      .6
       0       7
      .6      .6
       0       7
Pier Skew, UpSta & Num, DnSta & Num=  ,79, 2 ,63.5, 2 , 0 , 0 , 0 ,,
      .6      .6
       0       7
      .6      .6
       0       7
BR Coef=-1 , 0 , 0 ,, 0 ,,,0.8,-1,,0,
WSPro=,,,, 1 ,,,, 0 ,,,, 0 ,,,,-1 ,-1 ,-1 , 0 , 0 , 0 , 0 , 0
BC Design=,, 0 ,, 0 ,,,,,,

Type RM Length L Ch R = 1 ,30.38   ,24,24,24
#Sta/Elev= 21
       0     6.8    39.5    6.58    39.5    5.98    40.1    5.98    40.1    4.69
    45.5    1.28      50    1.35      53    1.39      54    1.23    55.5       1
      59    1.01    59.5    1.23      60    1.41    63.5    1.39      71    1.39
    73.9    3.73    73.9    5.98    74.5    5.98    74.5    6.58      84    6.57
     127    6.39
#Mann= 3 , 0 , 0
       0     .03       0    39.5     .03       0    74.5     .03       0
Bank Sta=39.5,74.5
Exp/Cntr=0.5,0.3

Type RM Length L Ch R = 1 ,30.14   ,11,11,11
#Sta/Elev= 27
       0    7.38       0    7.36    16.6    6.86    18.1    6.58    19.3    7.27
    23.6       7    32.4    7.16    40.1    6.75    42.4    5.39    47.6    5.39
    50.3    3.66    53.9       2    56.4    1.31    64.3    1.23    64.6    1.03
    70.6    1.03    71.2    1.51    73.3    1.31    73.3    2.33    82.3    2.33
    82.3    1.26    83.3    1.26    88.4    3.78    94.6    6.55   101.6    6.55
   102.9    6.41   152.8    6.48
#Mann= 3 , 0 , 0
       0     .03       0    47.6     .03       0    94.6     .03       0
Bank Sta=47.6,94.6
Exp/Cntr=0.5,0.3

Type RM Length L Ch R = 3 ,30.085  ,,,
BEGIN DESCRIPTION:
ÁöÇÏÃ¶±³·®
END DESCRIPTION:
Bridge Culvert--1,0,-1,-1, 0
Deck Dist Width WeirC Skew NumUp NumDn MinLoCord MaxHiCord MaxSubmerge Is_Ogee
0.1,10,1.44,0, 2, 2, , , 0.95, 0, 0,0,,
       0     153
      10      10
      10      10
       0     153
      10      10
      10      10
Pier Skew, UpSta & Num, DnSta & Num=  ,54, 2 ,54, 2 , 0 , 0 , 0 ,,
     1.5     1.5
       0      10
     1.5     1.5
       0      10
Pier Skew, UpSta & Num, DnSta & Num=  ,78.6, 2 ,78.6, 2 , 0 , 0 , 0 ,,
     1.5     1.5
       0      10
     1.5     1.5
       0      10
BR Coef=-1 , 0 , 0 ,, 0 ,,,0.8,-1,,0,
WSPro=,,,, 1 ,,,, 0 ,,,, 0 ,,,,-1 ,-1 ,-1 , 0 , 0 , 0 , 0 , 0
BC Design=,, 0 ,, 0 ,,,,,,

Type RM Length L Ch R = 1 ,30.03   ,3,3,3
#Sta/Elev= 27
       0    7.38       0    7.36    16.6    6.86    18.1    6.58    19.3    7.27
    23.6       7    32.4    7.16    40.1    6.75    42.4    5.39    47.6    5.39
    50.3    3.66    53.9       2    56.4    1.31    64.3    1.23    64.6    1.03
    70.6    1.03    71.2    1.51    73.3    1.31    73.3    2.33    82.3    2.33
    82.3    1.26    83.3    1.26    88.4    3.78    94.6    6.55   101.6    6.55
   102.9    6.41   152.8    6.48
#Mann= 3 , 0 , 0
       0     .03       0    47.6     .03       0    94.6     .03       0
Bank Sta=47.6,94.6
Exp/Cntr=0.5,0.3

Type RM Length L Ch R = 1 ,30      ,50,50,50
#Sta/Elev= 19
       0    6.61    32.8    5.31    38.1     5.2    40.8    3.67      45    1.76
    54.8    1.34      55    1.23      56    1.13    60.3    1.08    61.3    1.23
    61.7    1.49    74.2     1.3    79.2    3.77      85    6.33    86.3    6.33
    88.1    6.48    90.1    6.48   126.8    6.08   156.8    6.08
#Mann= 3 , 0 , 0
       0     .03       0    38.1     .03       0      85     .03       0
Bank Sta=38.1,85
Exp/Cntr=0.3,0.1

Type RM Length L Ch R = 1 ,29      ,50,50,50
#Sta/Elev= 27
       0    5.62    32.5    5.77    42.5    5.95    51.4    8.07    58.5    8.07
      68    5.41    73.5    5.29    76.2     3.7      81    1.47      91     1.4
    91.3    1.22    91.8    1.17    97.3    1.17    97.8    1.22    98.1    1.45
      99    1.33     114     1.3   122.5    5.07   125.5    5.17   130.4    5.17
   130.7    4.86   131.4    4.86   132.5     5.5   145.2    5.62   150.5    7.17
   164.9    9.24     185    9.64
#Mann= 3 , 0 , 0
       0     .03       0    73.5     .03       0   122.5     .03       0
Bank Sta=73.5,122.5
Exp/Cntr=0.3,0.1

Type RM Length L Ch R = 1 ,28      ,12,12,12
#Sta/Elev= 25
       0    4.97      30    5.17    32.5    5.17    43.3    5.29    71.3    5.22
    73.8    3.82    78.5    1.46    93.5    1.45      94    1.21    94.5    1.11
    98.8    1.11   100.2    1.11   100.7    1.21     101    1.47   115.8    1.29
   120.9    3.67   123.8    5.17     125    5.17     127    5.17   129.4    5.17
   130.1    4.71   130.7    4.71   131.3     5.1   135.3     5.1   158.6    6.01
#Mann= 3 , 0 , 0
       0     .03       0    71.3     .03       0   123.8     .03       0
Bank Sta=71.3,123.8
Exp/Cntr=0.3,0.1

Type RM Length L Ch R = 1 ,27.38   ,30,30,30
#Sta/Elev= 28
       0    4.72    25.7    4.91    35.7    4.82      54    4.97      54       4
   54.85       4   54.85    3.63      56    3.63      61    1.23      71    1.23
      75    1.23    75.5     .92      76     .73    80.5     .73    82.5     .73
      83     .92    83.5    1.18      88    1.18      98    1.23     102    3.63
  103.15    3.63  103.15       4     104       4     104    4.99   125.8    4.94
   133.8    5.02   142.1    4.91     161     4.7
#Mann= 3 , 0 , 0
       0     .03       0      54     .03       0     104     .03       0
Bank Sta=54,104
Exp/Cntr=0.5,0.3

Type RM Length L Ch R = 3 ,27.23   ,,,
BEGIN DESCRIPTION:
È­Á¤11±³
END DESCRIPTION:
Bridge Culvert--1,0,-1,-1, 0
Deck Dist Width WeirC Skew NumUp NumDn MinLoCord MaxHiCord MaxSubmerge Is_Ogee
0.1,29,1.44,0, 2, 2, , , 0.95, 0, 0,0,,
      54     104
    4.97    4.99
       4       4
      54     104
    4.97    4.99
       4       4
Pier Skew, UpSta & Num, DnSta & Num=  ,71, 2 ,71, 2 , 0 , 0 , 0 ,,
       1       1
       0       5
       1       1
       0       5
Pier Skew, UpSta & Num, DnSta & Num=  ,88, 2 ,88, 2 , 0 , 0 , 0 ,,
       1       1
       0       5
       1       1
       0       5
BR Coef=-1 , 0 , 0 ,, 0 ,,,0.8,-1,,0,
WSPro=,,,, 1 ,,,, 0 ,,,, 0 ,,,,-1 ,-1 ,-1 , 0 , 0 , 0 , 0 , 0
BC Design=,, 0 ,, 0 ,,,,,,
